HEC-RAS study 021209_rocky_swamp.prj: Rocky Swamp

--- 021209_rocky_swamp.g01 (geometry) --- (continued)

Type RM Length L Ch R = 1 ,61522.7,499.8,499.8,499.8
BEGIN DESCRIPTION:
Rocky Swamp 122.0
END DESCRIPTION:
#Sta/Elev= 30
  4185.6  200.31  4225.6  199.32  4275.6  196.37  4295.6  195.82  4355.6  192.32
  4435.6  182.15  4555.6  162.38  4565.6   161.4  4595.6  161.24  4605.6  160.25
  4635.6  161.25  4765.6   159.5  4835.6   157.3  4855.6  158.68  4885.6  158.86
  4905.6  158.21  4945.6  159.66  4985.6  158.94  4988.9  158.37  4990.4  155.37
  5009.5  155.37    5011  158.37    5030  160.17    5090  160.12    5140  159.29
    5250  162.76    5260  162.58    5300  165.11    5360  166.35  5603.6  182.79
#Mann= 3 , 1 , 0
 4185.60    0.15       0  4988.9    0.05       0    5011    0.15       0
Bank Sta=4988.90,5011.00
Exp/Cntr=0.3,0.1

Type RM Length L Ch R = 1 ,61022.9,501.5,501.5,501.5
BEGIN DESCRIPTION:
Rocky Swamp 121.0
END DESCRIPTION:
#Sta/Elev= 30
    3974   201.5    4064  197.46    4104  196.82    4154  194.45    4324  182.03
    4344  181.22    4364  179.18    4444  174.45    4604  161.57    4714  158.96
    4734  159.45    4844  158.18    4904  158.89    4954   157.3    4964  158.79
    4974  159.05    4989  157.77  4990.5  154.77  5009.6  154.77  5011.1  157.77
    5070  159.21    5300  158.52    5350  159.45    5480  159.72    5510  161.44
    5530   163.7    5610  175.03    5640  180.69    5730   190.5  5798.1  194.49
#Mann= 3 , 1 , 0
 3974.00    0.15       0    4989    0.05       0  5011.1    0.15       0
Bank Sta=4989.00,5011.10
Exp/Cntr=0.3,0.1

Type RM Length L Ch R = 1 ,60521.4,499.9,499.9,499.9
BEGIN DESCRIPTION:
Rocky Swamp 120.0
END DESCRIPTION:
#Sta/Elev= 30
  4055.4  195.32  4125.4   189.9  4255.4  184.41  4285.4  183.65  4335.4  180.66
  4475.4  164.18  4525.4   161.3  4675.4   157.4  4695.4  158.06  4845.4  158.05
  4865.4  157.34  4955.4  157.47  4975.4  156.48    4989  157.17  4990.5  154.17
  5009.6  154.17  5011.1  157.17    5060  157.74    5130  156.78    5160  157.36
    5200  156.36    5250  157.55    5270     157    5310  157.72    5320  158.36
    5350  162.12    5460  180.53    5500  185.77    5530  188.59  5641.4   191.5
#Mann= 3 , 1 , 0
 4055.40    0.15       0    4989    0.05       0  5011.1    0.15       0
Bank Sta=4989.00,5011.10
Exp/Cntr=0.3,0.1

Type RM Length L Ch R = 1 ,60021.5,500.3,500.3,500.3
BEGIN DESCRIPTION:
Rocky Swamp 119.0
END DESCRIPTION:
#Sta/Elev= 30
  3768.1  196.46  3838.1  192.43  3868.1     189  4008.1  183.72  4098.1  181.88
  4188.1  170.05  4258.1   163.1  4388.1  158.58  4458.1  157.33  4608.1  157.04
  4618.1  156.45  4648.1  157.43  4987.9  156.57  4989.4  153.57  5010.6  153.57
  5012.1  156.57    5090  157.16    5100   158.2    5150  157.55    5170  156.01
    5280  159.47    5330  166.89    5380  171.08    5460  175.67    5500  178.95
    5570  186.41    5650  192.64    5690  194.57    5750  199.27  5795.8  201.13
#Mann= 3 , 1 , 0
 3768.10   0.141       0  4987.9    0.05       0  5012.1   0.141       0
Bank Sta=4987.90,5012.10
Exp/Cntr=0.3,0.1

Type RM Length L Ch R = 1 ,59521.2,500.2,500.2,500.2
BEGIN DESCRIPTION:
Rocky Swamp 118.0
END DESCRIPTION:
#Sta/Elev= 30
  3809.2  180.94  3899.2  181.01  3989.2  178.81  4019.2  177.14  4129.2  167.61
  4249.2   163.3  4269.2  163.56  4369.2  160.46  4469.2  160.47  4559.2  158.91
  4599.2  156.66  4609.2  157.51  4669.2  157.03  4699.2  157.86  4759.2  156.48
  4819.2  158.13  4939.2  155.63  4987.9  155.97  4989.4  152.97  5010.6  152.97
  5012.1  155.97    5070  154.92    5330  160.66    5440  168.98    5470  172.61
    5500  180.31    5540  186.58    5630  192.24    5650  191.73  5678.2  192.95
#Mann= 3 , 1 , 0
 3809.20   0.141       0  4987.9    0.05       0  5012.1   0.141       0
Bank Sta=4987.90,5012.10
Exp/Cntr=0.3,0.1

Type RM Length L Ch R = 1 ,59021.0,499.2,499.2,499.2
BEGIN DESCRIPTION:
Rocky Swamp 117.0
END DESCRIPTION:
#Sta/Elev= 30
  3835.5  180.66  3895.5  180.24  3965.5  177.65  4005.5  174.28  4075.5  170.41
  4235.5     166  4245.5  164.99  4375.5  162.63  4505.5   162.5  4525.5  161.63
  4685.5  162.77  4775.5  159.06  4975.5  156.78  4987.9  155.36  4989.4  152.36
  5010.6  152.36  5012.1  155.36    5020  156.09    5070  154.55    5210  156.35
    5680  154.13    5800   154.4    5850  155.53    5880  157.05    5900   159.6
    5930  164.91    6000   179.8    6040   185.7    6100  192.87  6127.2  194.82
#Mann= 3 , 1 , 0
 3835.50   0.141       0  4987.9    0.05       0  5012.1   0.141       0
Bank Sta=4987.90,5012.10
Exp/Cntr=0.3,0.1

Type RM Length L Ch R = 1 ,58521.8,501,501,501
BEGIN DESCRIPTION:
Rocky Swamp 116.0
END DESCRIPTION:
#Sta/Elev= 30
  3634.7  181.37  3684.7  180.02  3764.7  179.01  3834.7   175.3  3854.7   173.6
  3874.7  173.84  4014.7  169.67  4074.7  169.53  4484.7  163.97  4504.7  164.63
  4694.7  162.13  4774.7  162.66  4864.7  160.42  4944.7  154.85  4987.9  154.76
  4989.4  151.76  5010.6  151.76  5012.1  154.76    5590  154.16    5600  153.47
    5610  153.91    5660  163.58    5690  171.21    5730  179.06    5770  183.81
    5790  185.04    5810  187.47    5870  190.12    5890  191.99  5992.4  194.68
#Mann= 3 , 1 , 0
 3634.70    0.15       0  4987.9    0.05       0  5012.1    0.15       0
Bank Sta=4987.90,5012.10
Exp/Cntr=0.3,0.1

Type RM Length L Ch R = 1 ,58020.8,500.6,500.6,500.6
BEGIN DESCRIPTION:
Rocky Swamp 115.0
END DESCRIPTION:
#Sta/Elev= 30
  3288.1  182.59  3478.1  176.82  3528.1  176.12  3588.1   173.6  3668.1  172.72
  3738.1  169.09  3768.1  168.75  3828.1  166.01  4018.1  163.75  4048.1  164.64
  4268.1  164.41  4438.1  161.24  4468.1  162.56  4548.1  158.17  4858.1  153.27
  4878.1  154.07  4987.9  154.09  4989.4  151.09  5010.6  151.09  5012.1  154.09
    5460   154.1    5530  156.32    5580  159.64    5600     162    5640  169.08
    5670  170.84    5710  171.04    5810   179.1    5920  197.04  5940.7  198.28
#Mann= 3 , 1 , 0
 3288.10    0.15       0  4987.9    0.05       0  5012.1    0.15       0
Bank Sta=4987.90,5012.10
Exp/Cntr=0.3,0.1

Type RM Length L Ch R = 1 ,57520.2,500.8,500.8,500.8
BEGIN DESCRIPTION:
Rocky Swamp 114.0
END DESCRIPTION:
#Sta/Elev= 30
  3889.5  182.67  3909.5  182.22  4009.5  176.19  4069.5   174.5  4149.5  170.26
  4269.5  167.52  4359.5  166.61  4469.5  168.42  4539.5  168.67  4659.5  167.18
  4759.5  160.67  4769.5  160.33  4829.5  154.12  4987.9   153.9  4989.4   150.9
  5010.6   150.9  5012.1   153.9    5200  153.83    5210  156.57    5220  158.17
    5230  161.22    5240  164.82    5250  167.46    5260  171.05    5310  184.52
    5320  187.95    5370  195.53    5400  198.21    5460  200.21    5485  199.92
#Mann= 3 , 1 , 0
 3889.50    0.15       0  4987.9    0.05       0  5012.1    0.15       0
Bank Sta=4987.90,5012.10
Exp/Cntr=0.3,0.1

Type RM Length L Ch R = 1 ,57019.4,455.7,455.7,455.7
BEGIN DESCRIPTION:
Rocky Swamp 113.0
END DESCRIPTION:
#Sta/Elev= 30
  4039.8   182.2  4059.8  182.19  4169.8  174.61  4199.8  171.98  4289.8  166.87
  4369.8  165.01  4379.8     164  4439.8  163.85  4449.8  163.14  4499.8  162.77
  4519.8   163.2  4599.8  159.65  4609.8  159.64  4629.8  160.64  4819.8  155.03
  4839.8  153.86  4987.9   153.7  4989.4   150.7  5010.6   150.7  5012.1   153.7
    5120  153.77    5180  165.23    5190  166.63    5220  169.59    5270  172.52
    5350  175.16    5400  178.51    5440  180.28    5450  181.38  5502.1  184.07
#Mann= 3 , 1 , 0
 4039.80    0.15       0  4987.9    0.05       0  5012.1    0.15       0
Bank Sta=4987.90,5012.10
Exp/Cntr=0.3,0.1

Type RM Length L Ch R = 1 ,56563.7,546.1,546.1,546.1
BEGIN DESCRIPTION:
Rocky Swamp 112.0
END DESCRIPTION:
#Sta/Elev= 21
  4695.3  172.17  4755.3  171.64  4885.3  165.45  4925.3  156.14  4985.3  152.58
  4987.9  151.02  4989.4  148.02  5010.6  148.02  5012.1  151.02  5053.5   151.7
  5073.5  150.77  5093.5  150.42  5103.5   149.7  5123.5  150.46  5153.5  150.61
  5173.5  152.68  5223.5  161.71  5263.5  170.85  5273.5  172.69  5443.5  181.84
  5447.5  182.23
#Mann= 3 , 1 , 0
 4695.30    0.15       0  4987.9    0.05       0  5012.1    0.15       0
Bank Sta=4987.90,5012.10
Exp/Cntr=0.3,0.1

Type RM Length L Ch R = 1 ,56017.6,501.5,501.5,501.5
BEGIN DESCRIPTION:
Rocky Swamp 111.0
END DESCRIPTION:
#Sta/Elev= 27
  4671.8  171.27  4691.8  170.37  4721.8  170.28  4731.8  168.86  4781.8  166.26
  4791.8  166.12  4861.8  160.66  4871.8  160.24  4987.9  146.41  4989.4  143.41
  5010.6  143.41  5012.1  146.41    5020  147.21    5030  148.54    5050  149.28
    5060  148.92    5080  149.63    5120  155.65    5140  157.73    5220   166.7
    5240  167.59    5280  172.46    5360     179    5430  181.24    5440  182.05
    5450  182.19  5455.9  182.69
#Mann= 3 , 1 , 0
 4671.80    0.15       0  4987.9    0.05       0  5012.1    0.15       0
Bank Sta=4987.90,5012.10
Exp/Cntr=0.3,0.1

Type RM Length L Ch R = 1 ,55516.1,499.9,499.9,499.9
BEGIN DESCRIPTION:
Rocky Swamp 110.0
END DESCRIPTION:
#Sta/Elev= 26
  4587.4  173.43  4607.4  172.51  4697.4  168.71  4727.4  166.02  4767.4  163.71
  4787.4  161.87  4807.4  160.54  4827.4   158.3  4867.4  152.07  4887.4  150.01
  4927.4  149.81  4957.4  147.98  4977.4     146  4987.9  145.59  4989.4  142.59
  5010.6  142.59  5012.1  145.59    5020  148.53    5030  148.98    5080  149.34
    5110  150.78    5180  153.47    5340  165.78    5370  167.21    5440  173.26
  5512.2  181.62
#Mann= 3 , 1 , 0
 4587.40    0.15       0  4987.9    0.05       0  5012.1    0.15       0
Bank Sta=4987.90,5012.10
Exp/Cntr=0.3,0.1

Type RM Length L Ch R = 1 ,55016.2,564.7,564.7,564.7
BEGIN DESCRIPTION:
Rocky Swamp 109.0
END DESCRIPTION:
#Sta/Elev= 30
  4311.7  172.29  4321.7  171.66  4341.7  172.13  4481.7  168.21  4511.7  165.93
  4601.7  163.26  4651.7     159  4731.7  154.82  4771.7  154.66  4871.7  151.54
  4881.7  150.39  4911.7  150.34  4951.7   147.7  4981.7  146.68  4987.9  144.53
  4989.4  141.53  5010.6  141.53  5012.1  144.53    5020  148.35    5100  148.43
    5210  150.47    5270  152.52    5300  154.53    5360  157.09    5400  160.19
    5430  163.48    5470  166.32    5490  168.74    5540  172.26  5616.1  181.28
#Mann= 3 , 1 , 0
 4311.70    0.15       0  4987.9    0.05       0  5012.1    0.15       0
Bank Sta=4987.90,5012.10
Exp/Cntr=0.3,0.1

Type RM Length L Ch R = 1 ,54451.5,368.1,368.1,368.1
BEGIN DESCRIPTION:
Rocky Swamp 108.0
END DESCRIPTION:
#Sta/Elev= 30
    3991  173.61    4121  166.22    4191  163.06    4331  160.73    4381  157.98
    4401  158.35    4481  156.37    4501  155.18    4531  155.86    4571  154.12
    4611  153.68    4641  151.12    4691  149.52    4731  149.68    4761  148.47
    4941  145.92    4961  147.29    4981  147.14  4987.9  144.25  4989.4  141.25
  5010.6  141.25  5012.1  144.25  5018.1  147.36  5158.1   148.8  5168.1  149.76
  5228.1  159.81  5268.1  167.26  5308.1  171.59  5378.1  174.85  5462.3   175.1
#Mann= 3 , 1 , 0
 3991.00   0.141       0  4987.9    0.05       0  5012.1   0.141       0
Bank Sta=4987.90,5012.10
Exp/Cntr=0.3,0.1

Type RM Length L Ch R = 1 ,54083.4,571.2,571.2,571.2
BEGIN DESCRIPTION:
Rocky Swamp 107.0
END DESCRIPTION:
#Sta/Elev= 30
    3998  178.22    4058  175.58    4198  164.02    4318  160.41    4358  157.64
    4408  158.27    4508  156.83    4548   158.1    4588  156.72    4638  157.68
    4668   155.9    4718  149.36    4838  147.16    4958  147.76  4987.9  143.67
  4989.4  140.67  5010.6  140.67  5012.1  143.67    5016  145.87    5086  147.18
    5116   147.1    5136  146.05    5256  147.55    5276  147.03    5356  148.43
    5486  158.81    5536  159.99    5606  168.21    5736  179.03  5827.4  182.46
#Mann= 3 , 1 , 0
 3998.00   0.141       0  4987.9    0.05       0  5012.1   0.141       0
Bank Sta=4987.90,5012.10
Exp/Cntr=0.3,0.1

Type RM Length L Ch R = 1 ,53512.2,499.5,499.5,499.5
BEGIN DESCRIPTION:
Rocky Swamp 106.0
END DESCRIPTION:
#Sta/Elev= 30
  3924.3  173.66  3994.3   171.9  4014.3  170.07  4044.3  169.64  4064.3  167.61
  4174.3  163.35  4184.3  162.45  4194.3  159.51  4214.3  162.02  4334.3  162.41
  4404.3  160.69  4434.3  161.56  4624.3  160.08  4714.3   158.5  4744.3   156.9
  4794.3  156.82  4834.3  154.31  4894.3   152.9  4914.3  149.48  4944.3  146.34
  4984.3  145.24  4987.9  142.56  4989.4  139.56  5010.6  139.56  5012.1  142.56
    5020  145.15    5110  146.74    5390  146.96    5430   148.3  5850.6  172.69
#Mann= 3 , 1 , 0
 3924.30   0.141       0  4987.9    0.05       0  5012.1   0.141       0
Bank Sta=4987.90,5012.10
Exp/Cntr=0.3,0.1

Type RM Length L Ch R = 1 ,53012.7,499.9,499.9,499.9
BEGIN DESCRIPTION:
Rocky Swamp 105.0
END DESCRIPTION:
#Sta/Elev= 30
  4043.2  184.16  4083.2  181.25  4183.2  176.07  4313.2  162.82  4423.2  158.87
  4443.2  159.11  4503.2  156.43  4543.2   156.7  4563.2  155.76  4723.2  155.61
  4843.2   157.5  4863.2  157.01  4943.2  147.83  4963.2  144.32    4985  142.33
  4986.5  139.33  5013.6  139.33  5015.1  142.33    5020  144.54    5050  146.12
    5170  144.87    5330   146.9    5380     146    5750  147.06    5850  155.44
    5920  157.57    5960  160.06    6030  168.26    6110  175.21  6164.7  177.12
#Mann= 3 , 1 , 0
 4043.20   0.141       0    4985    0.05       0  5015.1   0.141       0
Bank Sta=4985.00,5015.10
Exp/Cntr=0.3,0.1

Type RM Length L Ch R = 1 ,52512.8,500.9,500.9,500.9
BEGIN DESCRIPTION:
Rocky Swamp 104.0
END DESCRIPTION:
#Sta/Elev= 30
  4049.6  184.47  4139.6  180.53  4269.6  170.97  4409.6   158.5  4579.6   153.4
  4709.6   154.7  4779.6  157.55  4869.6   156.8  4899.6  153.37  4929.6  147.02
    4985  142.14  4986.5  139.14  5013.6  139.14  5015.1  142.14    5020  144.35
    5040  144.96    5110  145.15    5120   142.9    5180  146.01    5290  145.58
    5310   147.5    5340  147.89    5450  145.46    5500  146.52    5770  144.51
    5930  145.78    6020  152.87    6120  167.42    6180  169.59  6244.8  174.45
#Mann= 3 , 1 , 0
 4049.60   0.141       0    4985    0.05       0  5015.1   0.141       0
Bank Sta=4985.00,5015.10
Exp/Cntr=0.3,0.1

Type RM Length L Ch R = 1 ,52011.9,1001.3,1001.3,1001.3
BEGIN DESCRIPTION:
Rocky Swamp 103.0
END DESCRIPTION:
#Sta/Elev= 30
  3952.4   182.9  4012.4  179.51  4042.4  176.74  4062.4  176.49  4112.4  172.27
  4142.4  171.11  4172.4  168.01  4282.4  159.74  4362.4  156.26  4462.4  153.83
  4582.4  153.13  4762.4  147.73  4932.4  146.75    4985  141.95  4986.5  138.95
  5013.6  138.95  5015.1  141.95    5070  144.55    5090  143.42    5250   145.1
    5300   143.8    5360  145.68    5490  143.03    5570  144.92    5670  144.95
    5730  146.43    5770  150.55    5830  162.96    5930  172.35  5965.4   172.8
#Mann= 3 , 1 , 0
 3952.40   0.141       0    4985    0.05       0  5015.1   0.141       0
Bank Sta=4985.00,5015.10
Exp/Cntr=0.3,0.1

Type RM Length L Ch R = 1 ,51010.6,500.6,500.6,500.6
BEGIN DESCRIPTION:
Rocky Swamp 102.0
END DESCRIPTION:
#Sta/Elev= 30
  3840.4  182.41  3930.4  179.43  4110.4   168.3  4150.4  164.03  4230.4  158.53
  4330.4  153.05  4460.4   151.2  4590.4  145.93  4660.4  145.64  4710.4  143.57
  4750.4  144.12  4790.4  142.52  4910.4  144.91  4980.4  144.42  4984.9   141.5
  4986.4   138.5  5013.5   138.5    5015   141.5    5040  143.14    5110  143.75
    5230   144.1    5250  142.99    5370  144.83    5490  143.94    5580  145.13
    5820  145.05    5850  146.49    5880  153.54    5980  168.62  6080.3  174.76
#Mann= 3 , 1 , 0
 3840.40   0.141       0  4984.9    0.05       0    5015   0.141       0
Bank Sta=4984.90,5015.00
Exp/Cntr=0.3,0.1

Type RM Length L Ch R = 1 ,50510.0,501.4,501.4,501.4
BEGIN DESCRIPTION:
Rocky Swamp 101.0
END DESCRIPTION:
#Sta/Elev= 30
  3887.6  176.32  3977.6  173.31  4067.6   165.9  4197.6  159.62  4227.6   157.1
  4437.6  149.22  4457.6  149.86  4607.6  147.83  4677.6  145.06  4797.6  144.11
  4837.6  142.06  4947.6  142.82  4984.9  138.88  4986.4  135.88  5013.6  135.88
  5015.1  138.88    5040  142.97    5070  143.51    5340  142.59    5400  145.44
    5450  143.79    5530  143.71    5580  145.04    5720  145.41    5900  148.89
    6050  159.81    6100  157.96    6260  163.31    6460  182.01  6531.5  185.45
#Mann= 3 , 1 , 0
 3887.60   0.141       0  4984.9    0.05       0  5015.1   0.141       0
Bank Sta=4984.90,5015.10
Exp/Cntr=0.3,0.1

Type RM Length L Ch R = 1 ,50008.6,499,499,499
BEGIN DESCRIPTION:
Rocky Swamp 100.0
END DESCRIPTION:
#Sta/Elev= 30
    3531  173.82    3641  166.23    3801  159.32    3931  158.41    3971  156.57
    4031  151.51    4091  148.82    4411  143.55    4591  141.95    4871  143.08
    4901   144.1    4951   142.2    4985  137.96  4986.5  134.96  5013.6  134.96
  5015.1  137.96    5030  141.18    5070  141.09    5090  142.44    5150     141
    5180  142.74    5310  143.63    5340  145.62    5500  144.17    5670  147.66
    5720  151.64    5840  169.17    5860  170.93    6080  172.38  6257.7  184.29
#Mann= 3 , 1 , 0
 3531.00   0.141       0    4985    0.05       0  5015.1   0.141       0
Bank Sta=4985.00,5015.10
Exp/Cntr=0.3,0.1

Type RM Length L Ch R = 1 ,49509.6,498.3,498.3,498.3
BEGIN DESCRIPTION:
Rocky Swamp 99.0
END DESCRIPTION:
#Sta/Elev= 30
  3345.1  174.84  3415.1  170.11  3465.1  168.07  3515.1  168.67  3625.1  164.29
  3685.1  160.12  3815.1  155.75  3905.1     156  4015.1   149.2  4105.1  145.49
  4265.1  142.35  4415.1  141.26  4465.1  142.11  4925.1  141.57  4945.1  142.63
  4975.1  142.22  4984.9  137.35  4986.4  134.35  5013.6  134.35  5015.1  137.35
    5040  141.73    5090  142.85    5300  141.01    5400  141.62    5470  147.45
    5520  148.93    5560  151.86    5710  166.77    5730  169.81  5781.1   172.7
#Mann= 3 , 1 , 0
 3345.10   0.141       0  4984.9    0.05       0  5015.1   0.141       0
Bank Sta=4984.90,5015.10
Exp/Cntr=0.3,0.1

Type RM Length L Ch R = 1 ,49011.3,502.4,502.4,502.4
BEGIN DESCRIPTION:
Rocky Swamp 98.0
END DESCRIPTION:
#Sta/Elev= 30
  3427.8  174.51  3477.8  169.19  3627.8  163.14  3817.8  157.93  3867.8  155.76
  3927.8  154.82  4267.8   141.3  4367.8   140.9  4427.8  141.78  4617.8   139.3
  4687.8  141.17  4927.8  140.48  4984.9  136.73  4986.4  133.73  5013.6  133.73
  5015.1  136.73    5020  139.75    5050     141    5160  139.13    5190  140.33
    5230  139.66    5260  141.88    5350   141.4    5390  142.22    5450  146.51
    5500  153.19    5550  158.47    5740  170.56    5780  172.41  5792.1  172.16
#Mann= 3 , 1 , 0
 3427.80    0.15       0  4984.9   0.055       0  5015.1    0.15       0
Bank Sta=4984.90,5015.10
Exp/Cntr=0.3,0.1

Type RM Length L Ch R = 1 ,48508.9,297.6,297.6,297.6
BEGIN DESCRIPTION:
Rocky Swamp 97.0
END DESCRIPTION:
#Sta/Elev= 30
  3571.3  168.55  3651.3  165.18  3721.3  163.55  3961.3   151.2  4141.3  146.79
  4201.3  143.87  4351.3  142.23  4521.3  139.42  4591.3  140.05  4651.3  138.65
  4931.3  139.89  4971.3  138.64  4984.9  135.67  4986.4  132.67  5013.5  132.67
    5015  135.67    5050  139.57    5140  139.86    5170  139.27    5190  139.85
    5290  139.95    5320  140.83    5600  140.33    5670  144.27    5710   149.8
    5780   164.8    5800   168.1    5820  172.31    5870  179.28  5909.6  182.61
#Mann= 3 , 1 , 0
 3571.30    0.15       0  4984.9   0.055       0    5015    0.15       0
Bank Sta=4984.90,5015.00
Exp/Cntr=0.3,0.1

Type RM Length L Ch R = 1 ,48211.3,817.7,817.7,817.7
BEGIN DESCRIPTION:
Rocky Swamp 96.0
END DESCRIPTION:
#Sta/Elev= 30
  4241.5  146.27  4321.5   144.9  4341.5  143.76  4351.5  144.24  4381.5  142.86
  4411.5  140.44  4531.5  138.99  4661.5   140.3  4741.5  139.61  4761.5  138.35
  4791.5  138.11  4821.5  139.49  4861.5  138.89  4911.5  139.82  4931.5  139.22
  4961.5  140.17  4984.9  135.55  4986.4  132.55  5013.5  132.55    5015  135.55
  5015.3  140.23  5055.3  140.49  5205.3  138.82  5445.3  139.45  5475.3   140.3
  5505.3  143.15  5565.3  152.65  5665.3  166.83  5725.3  172.71  5740.6   173.3
#Mann= 3 , 1 , 0
 4241.50    0.15       0  4984.9   0.055       0    5015    0.15       0
Bank Sta=4984.90,5015.00
Exp/Cntr=0.3,0.1

Type RM Length L Ch R = 1 ,47393.6,387.6,387.6,387.6
BEGIN DESCRIPTION:
Rocky Swamp 95.0
END DESCRIPTION:
#Sta/Elev= 30
  3748.3  173.15  3818.3  169.49  3848.3  166.94  3908.3  159.62  3958.3  155.96
  4088.3  149.99  4128.3  145.66  4168.3  143.06  4208.3  139.18  4278.3  137.88
  4348.3  138.81  4698.3  138.42  4918.3  139.62  4958.3   138.4  4983.8  134.04
  4985.3  131.04  5014.8  131.04  5016.3  134.04  5055.4  140.35  5125.4  142.81
  5145.4  140.61  5175.4  141.73  5215.4  145.04  5235.4  148.08  5255.4  145.98
  5305.4  146.53  5335.4  147.88  5435.4  163.78  5565.4  174.33  5603.7  175.16
#Mann= 3 , 1 , 0
 3748.30    0.15       0  4983.8   0.055       0  5016.3    0.15       0
Bank Sta=4983.80,5016.30
Exp/Cntr=0.3,0.1

Type RM Length L Ch R = 1 ,47006.0,275.5,275.5,275.5
BEGIN DESCRIPTION:
Rocky Swamp 94.0
END DESCRIPTION:
#Sta/Elev= 30
  3688.1  177.76  3798.1  173.26  3808.1  172.45  3828.1  168.73  3888.1  164.77
  3958.1  157.79  4178.1  148.92  4188.1  148.88  4338.1   139.2  4408.1  137.97
  4538.1   137.7  4548.1  138.46  4598.1     138  4618.1  136.82  4658.1  137.43
  4718.1  135.92  4768.1  137.72  4938.1  138.59  4958.1  137.73  4983.7  133.39
  4985.2  130.39  5014.7  130.39  5016.2  133.39    5040  137.68    5050   138.6
    5160   138.2    5180  138.96    5220  144.15    5280     160  5320.3  163.24
#Mann= 3 , 1 , 0
 3688.10    0.15       0  4983.7   0.055       0  5016.2    0.15       0
Bank Sta=4983.70,5016.20
Exp/Cntr=0.3,0.1

Type RM Length L Ch R = 1 ,46730.5,722.6,722.6,722.6
BEGIN DESCRIPTION:
Rocky Swamp 93.0
END DESCRIPTION:
#Sta/Elev= 30
  3816.2  173.95  3856.2  169.55  3986.2   160.2  3996.2  159.01  4096.2   152.4
  4376.2  144.63  4436.2  141.43  4446.2  141.71  4476.2  140.17  4566.2  140.22
  4686.2  138.14  4796.2  139.45  4876.2  137.07  4916.2  137.77  4936.2  135.69
  4956.2  134.77  4976.2  135.04  4983.7  132.93  4985.2  129.93  5014.7  129.93
  5016.2  132.93  5020.9  134.65  5040.9  135.27  5080.9  137.83  5220.9  138.14
  5230.9   139.1  5260.9  146.78  5350.9  160.81  5440.9  166.18    5494  166.79
#Mann= 3 , 1 , 0
 3816.20    0.15       0  4983.7   0.055       0  5016.2    0.15       0
Bank Sta=4983.70,5016.20
Exp/Cntr=0.3,0.1

Type RM Length L Ch R = 1 ,46007.9,354.5,354.5,354.5
BEGIN DESCRIPTION:
Rocky Swamp 92.0
END DESCRIPTION:
#Sta/Elev= 30
  3937.9   163.9  3977.9  161.59  4107.9  156.68  4127.9  155.25  4197.9  153.07
  4217.9  153.56  4237.9  152.01  4307.9  149.82  4327.9  150.26  4347.9  148.76
  4437.9  147.04  4507.9     142  4527.9     142  4697.9  137.02  4857.9  138.15
  4957.9  137.46  4983.8  132.72  4985.3  129.72  5014.8  129.72  5016.3  132.72
    5020  136.73    5030  137.33    5350  137.11    5520  137.77    5530  138.36
    5590  146.01    5620  151.95    5680   165.3    5720  171.28  5763.7  175.59
#Mann= 3 , 1 , 0
 3937.90    0.15       0  4983.8   0.055       0  5016.3    0.15       0
Bank Sta=4983.80,5016.30
Exp/Cntr=0.3,0.1

Type RM Length L Ch R = 1 ,45653.4,650.2,650.2,650.2
BEGIN DESCRIPTION:
Rocky Swamp 91.0
END DESCRIPTION:
#Sta/Elev= 30
  3833.7  162.02  3893.7  159.85  3903.7  160.35  3943.7  157.52  4103.7  151.92
  4123.7   152.4  4363.7  149.27  4503.7  145.67  4513.7  145.12  4523.7  142.84
  4553.7  139.11  4603.7  136.13  4883.7  136.56  4923.7   137.5  4963.7  136.19
  4983.8  131.93  4985.3  128.93  5014.7  128.93  5016.2  131.93  5030.8  139.52
  5106.9  143.38  5210.8  136.28  5290.8  137.69  5310.8  139.05  5370.8  146.66
  5400.8  152.27  5430.8  154.95  5450.8  155.83  5510.8   154.9  5673.2  162.54
#Mann= 4 , 1 , 0
 3833.70    0.15       0  4983.8   0.055       0  5016.2    0.15       0
  5106.9       1       0
Bank Sta=4983.80,5016.20
Exp/Cntr=0.3,0.1

Type RM Length L Ch R = 1 ,45003.2,498.3,498.3,498.3
BEGIN DESCRIPTION:
Rocky Swamp 90.0
END DESCRIPTION:
#Sta/Elev= 30
    3908  164.48    3938  162.63    3978  158.39    4008  157.87    4048  155.61
    4148  154.37    4298  147.58    4358  146.31    4368  147.28    4418  145.69
    4528  145.44    4578  141.84    4608  140.76    4658  136.42    4978  135.37
  4983.8  131.02  4985.3  128.02  5014.8  128.02  5016.3  131.02    5070  135.08
    5120  135.39    5150  134.28    5280  136.75    5330  136.12    5360  137.37
    5520  138.03    5560  140.34    5600  145.18    5680   163.1  5689.3  164.44
#Mann= 3 , 1 , 0
 3908.00    0.15       0  4983.8   0.055       0  5016.3    0.15       0
Bank Sta=4983.80,5016.30
Exp/Cntr=0.3,0.1

Type RM Length L Ch R = 1 ,44504.9,499.8,499.8,499.8
BEGIN DESCRIPTION:
Rocky Swamp 89.0
END DESCRIPTION:
#Sta/Elev= 30
  3919.6  164.58  3979.6  159.92  4119.6  154.51  4149.6  149.98  4169.6  145.59
  4219.6  139.68  4339.6  136.27  4359.6  137.66  4449.6   137.7  4539.6  135.45
  4689.6  137.37  4729.6  136.52  4769.6  138.13  4799.6  137.95  4889.6  132.87
  4939.6  135.86  4969.6  136.06  4983.7  130.73  4985.2  127.73  5014.7  127.73
  5016.2  130.73    5050  135.63    5460  135.36    5500  140.64    5570   155.9
    5580   157.2    5640  162.29    5660  163.02    5670  164.52  5715.4  166.24
#Mann= 3 , 1 , 0
 3919.60    0.15       0  4983.7   0.055       0  5016.2    0.15       0
Bank Sta=4983.70,5016.20
Exp/Cntr=0.3,0.1

Type RM Length L Ch R = 1 ,44005.1,500.2,500.2,500.2
BEGIN DESCRIPTION:
Rocky Swamp 88.0
END DESCRIPTION:
#Sta/Elev= 30
  4082.3  172.55  4222.3   163.2  4302.3  158.99  4322.3  156.93  4372.3  154.67
  4512.3  136.05  4892.3  134.67  4922.3  131.12  4952.3  133.86  4962.3  133.16
  4972.3  135.19  4982.3  134.21  4983.7  129.36  4985.2  126.36  5014.7  126.36
  5016.2  129.36    5040  131.31    5110  131.29    5160  134.89    5290  135.18
    5370  134.37    5390  135.06    5700  135.39    5750  136.36    5800  139.14
    5870  147.61    5910   157.8    5950  165.78    6000   169.8    6043  169.94
#Mann= 3 , 1 , 0
 4082.30    0.15       0  4983.7   0.055       0  5016.2    0.15       0
Bank Sta=4983.70,5016.20
Exp/Cntr=0.3,0.1

Type RM Length L Ch R = 1 ,43504.9,501.8,501.8,501.8
BEGIN DESCRIPTION:
Rocky Swamp 87.0
END DESCRIPTION:
#Sta/Elev= 30
  4159.8  165.57  4289.8  158.04  4359.8  152.42  4399.8  151.88  4439.8  148.75
  4529.8  138.32  4589.8  134.65  4839.8  133.54  4899.8   135.1  4949.8  134.09
  4979.8  130.83  4983.7  129.21  4985.2  126.21  5014.7  126.21  5016.2  129.21
    5040  133.91    5160  134.62    5190  136.49    5210  138.94    5300   142.1
    5400  142.45    5440  144.28    5470  143.78    5490  145.78    5670  148.16
    5700  147.72    5840  157.08    5920  158.37    5960  157.99  6075.6  162.71
#Mann= 3 , 1 , 0
 4159.80   0.141       0  4983.7   0.055       0  5016.2   0.141       0
Bank Sta=4983.70,5016.20
Exp/Cntr=0.3,0.1

Type RM Length L Ch R = 1 ,43003.1,499.8,499.8,499.8
BEGIN DESCRIPTION:
Rocky Swamp 86.0
END DESCRIPTION:
#Sta/Elev= 30
  3869.9   172.2  4009.9   164.6  4039.9  161.54  4119.9  150.09  4179.9  145.59
  4229.9  143.01  4299.9  143.82  4379.9  139.05  4449.9  136.67  4469.9  135.02
  4619.9  133.37  4799.9  134.42  4969.9  133.78  4983.8  129.05  4985.3  126.05
  5014.7  126.05  5016.2  129.05    5110   134.7    5130  134.19    5180  138.29
    5250  138.67    5280  137.74    5370   140.3    5400  139.99    5410  140.97
    5500  141.51    5880   149.2    5930  154.09    6150  160.92  6204.8  163.56
#Mann= 3 , 1 , 0
 3869.90   0.141       0  4983.8   0.055       0  5016.2   0.141       0
Bank Sta=4983.80,5016.20
Exp/Cntr=0.3,0.1

Type RM Length L Ch R = 1 ,42503.3,500.5,500.5,500.5
BEGIN DESCRIPTION:
Rocky Swamp 85.0
END DESCRIPTION:
#Sta/Elev= 30
    3661  161.19    3721  159.22    3811  153.94    3851  154.62    3921  150.97
    4011  147.84    4091  144.11    4121  141.83    4311  136.02    4491  134.75
    4591  132.21    4661  132.46    4691  131.63    4731  133.76    4841  134.35
    4861  133.45    4951  133.22    4961  132.91  4983.8   128.5  4985.3   125.5
  5014.8   125.5  5016.3   128.5    5050  133.42    5250  138.63    5390  140.76
    5440  142.93    5660   148.9    5690  152.05    5800  155.03  5971.3  162.44
#Mann= 3 , 1 , 0
 3661.00   0.141       0  4983.8   0.055       0  5016.3   0.141       0
Bank Sta=4983.80,5016.30
Exp/Cntr=0.3,0.1

Type RM Length L Ch R = 1 ,42002.8,500.7,500.7,500.7
BEGIN DESCRIPTION:
Rocky Swamp 84.0
END DESCRIPTION:
#Sta/Elev= 30
  3867.9  173.37  3927.9  170.84  3977.9  165.61  3997.9  162.08  4087.9  150.96
  4117.9  148.37  4157.9  143.04  4197.9  139.61  4257.9  138.57  4287.9   136.6
  4447.9  133.32  4717.9  131.21  4757.9  132.52  4927.9  134.03  4977.9   132.3
  4983.8  127.75  4985.3  124.75  5014.7  124.75  5016.2  127.75    5030   132.3
    5090  130.36    5120  133.78    5190  132.61    5280     134    5310  136.31
    5400  138.35    5450  141.53    5660   145.9    5720  149.94  5973.2   163.4
#Mann= 3 , 1 , 0
 3867.90   0.141       0  4983.8   0.055       0  5016.2   0.141       0
Bank Sta=4983.80,5016.20
Exp/Cntr=0.3,0.1

Type RM Length L Ch R = 1 ,41502.1,499.9,499.9,499.9
BEGIN DESCRIPTION:
Rocky Swamp 83.0
END DESCRIPTION:
#Sta/Elev= 30
  4096.8  163.12  4146.8  159.05  4326.8  153.21  4366.8  153.23  4446.8  151.06
  4516.8   140.9  4556.8  133.31  4596.8  130.84  4706.8  133.31  4766.8  132.25
  4786.8     131  4906.8  133.56  4956.8  132.73  4976.8  129.91  4983.8  127.21
  4985.3  124.21  5014.7  124.21  5016.2  127.21    5020  130.73    5030   131.6
    5080  128.93    5110   132.3    5210  130.51    5270  133.24    5430  135.56
    5460  137.44    5730  145.72    5840  152.92    5910  158.92  5994.4  161.59
#Mann= 3 , 1 , 0
 4096.80   0.141       0  4983.8   0.055       0  5016.2   0.141       0
Bank Sta=4983.80,5016.20
Exp/Cntr=0.3,0.1

Type RM Length L Ch R = 1 ,41002.2,773.3,773.3,773.3
BEGIN DESCRIPTION:
Rocky Swamp 82.0
END DESCRIPTION:
#Sta/Elev= 30
  4088.2  165.57  4118.2  165.65  4148.2  163.45  4188.2  158.14  4278.2  140.28
  4298.2  137.25  4338.2  134.28  4448.2  134.34  4458.2   133.4  4728.2  130.09
  4938.2  131.24  4948.2     131  4983.8   126.8  4985.3   123.8  5014.8   123.8
  5016.3   126.8    5020  129.96    5040  131.69    5230  131.79    5240  131.13
    5290  131.87    5350  130.81    5410  131.77    5470  134.06    5500  136.45
    5810  141.85    5920  148.03    5960  149.09    6060  156.35  6207.9  161.26
#Mann= 3 , 1 , 0
 4088.20   0.141       0  4983.8   0.055       0  5016.3   0.141       0
Bank Sta=4983.80,5016.30
Exp/Cntr=0.5,0.3

Type RM Length L Ch R = 1 ,40228.9,45,45,45
BEGIN DESCRIPTION:
Upstream Section of Bridge/Culvert/Weir
END DESCRIPTION:
#Sta/Elev= 30
  4135.3  162.64  4181.2  152.76  4211.2  150.71  4311.2  147.92  4341.2  146.25
  4371.2  146.12  4381.2  144.99  4421.2  147.65  4431.2  147.43  4511.2  143.31
  4631.2  133.77  4711.2  129.16  4771.2  130.54  4841.2  129.11  4901.2  129.92
  4951.2  129.22  4979.5  127.06  4986.5  122.26  5013.5  122.26  5020.5  127.06
  5128.6  131.14  5248.6  131.62  5338.6  135.41  5398.6  136.34  5468.6   143.6
  5488.6   147.6  5608.6  146.55  6028.6  152.77  6298.6   161.3  6624.6  164.56
#Mann= 3 , 1 , 0
 4135.30   0.131       0  4979.5   0.055       0  5020.5   0.131       0
#XS Ineff= 2 , 0
       0    4920     136    5079       0     134
Bank Sta=4979.50,5020.50
Exp/Cntr=0.5,0.3

Type RM Length L Ch R = 3 ,40206.4,,,
BEGIN DESCRIPTION:
Ringwood Road-TOR
Structure ID: Ringwood Road
Approximate Survey Structure
END DESCRIPTION:
Bridge Culvert--1,0,-1,-1, 0
Deck Dist Width WeirC Skew NumUp NumDn MinLoCord MaxHiCord MaxSubmerge Is_Ogee
10,25,2.6,, 47, 48,,,0.95,0,1,1,,
  4135.3  4181.2  4201.2  4211.2  4225.3  4245.3  4265.3  4310.6  4321.2  4331.2
  4341.2  4371.2  4381.2  4401.2  4421.2  4431.2  4441.2  4511.2  4580.6  4601.2
  4621.2  4631.2  4711.2  4771.2  4790.6  4810.6  4841.2  4871.2  4881.2  4901.2
 4930.91    4931  4940.6 5068.89    5069  5108.6  5128.6  5248.6  5314.5  5338.6
  5398.6  5468.6  5488.6  5608.6  6028.6  6298.6  6624.6
  162.63  159.66  158.42   157.8  156.92  155.32  150.68  149.97  149.36   148.8
  148.56  147.86  147.63  147.16  147.64  147.42  146.39  144.19  142.31  141.87
  141.44  141.22  139.51  138.22   137.8  137.85  137.23  136.77  136.61   136.3
  135.84  135.84  135.69  135.26  135.26  135.13  135.06  134.66  134.39   135.4
  136.33  143.59  147.59  146.54  152.76  161.29  164.55
  162.63  152.75  151.64   150.7  150.23   149.6  149.08  147.93  147.21  147.06
  146.24  146.11  144.98  146.47  147.64  147.42  146.39   143.3  137.63  135.95
  134.87  133.76  129.15  130.53  130.13  129.73   129.1   129.6  129.32  129.91
  129.49  134.06  133.91  133.48  129.01  130.61  131.13  131.61  134.39   135.4
  136.33  143.59  147.59  146.54  152.76  161.29  164.55
  4135.3  4181.2  4201.2  4211.2  4225.3  4245.3  4265.3  4310.6  4321.2  4331.2
  4341.2  4371.2  4381.2  4401.2  4421.2  4431.2  4441.2  4511.2  4580.6  4601.2
  4621.2  4631.2  4711.2  4771.2  4790.6  4810.6  4841.2  4871.2  4881.2  4901.2
 4930.91    4931  4940.6 5068.89    5069  5108.6  5128.6  5248.6  5304.5  5314.5
  5338.6  5398.6  5468.6  5488.6  5608.6  6028.6  6298.6  6624.6
  162.51  159.66  158.42   157.8  156.92  155.32  150.68  149.97  149.36   148.8
  148.56  147.86  147.63  147.16  147.53  147.31  146.28  144.19  142.31  141.87
  141.44  141.22  139.51  138.22   137.8  137.85  137.23  136.77  136.61   136.3
  135.84  135.84  135.69  135.26  135.26  135.13  135.06  134.66  134.47  134.28
  135.29  136.28  143.48  147.48  146.43  152.65  161.18  164.43
  162.38   152.5  151.39  150.45  149.98  149.35  148.83  147.68  146.96  146.81
  145.99  145.86  144.73  146.22  147.39  147.17  146.14  143.05  137.38   135.7
  134.62  133.51   128.9  130.28  129.88  129.48  128.85  129.35  129.07  129.66
  129.24  133.81  133.66  133.23  128.76  130.36  130.88  131.36  133.71  134.14
  135.15  136.08  143.34  147.34  146.29  152.51  161.04   164.3
Pier Skew, UpSta & Num, DnSta & Num=,4983.7, 2 ,4983.7, 2 , 0 , 0 , 0 ,,
       2       2
  122.48  134.77
       2       2
  122.23  134.52
Pier Skew, UpSta & Num, DnSta & Num=,5016.2, 2 ,5016.2, 2 , 0 , 0 , 0 ,,
       2       2
  122.42  134.66
       2       2
  122.17  134.41
Abutment Skew #Up #Dn=, 2 , 2
 4930.80 4967.50
  134.06  127.97
 4930.80 4967.50
  133.81  127.72
Abutment Skew #Up #Dn=, 2 , 2
 5032.50 5069.09
  127.53  133.48
 5032.50 5069.09
  127.28  133.23
BR Coef= 1 , 1 , 0 ,1.25, 0 ,,,0.8,0,2,0,
Wspro=,,,, 1 ,,,, 0 ,,,, 0 ,,,,-1 ,-1 ,-1 , 0 , 0 , 0 , 0 , 0
BC Design=,, 0 ,, 0 ,,,,,,
BR U #Sta/Elev= 75
  4135.3  162.63  4181.2  152.75  4201.2  151.64  4211.2   150.7  4225.3  150.23
  4241.2   149.7  4245.3   149.6  4265.3  149.08  4310.6  147.93  4311.2  147.91
  4321.2  147.21  4330.6  147.07  4331.2  147.06  4341.2  146.24  4371.2  146.11
  4381.2  144.98  4400.6  146.43  4401.2  146.47  4421.2  147.64  4431.2  147.42
  4441.2  146.39  4511.2   143.3  4580.6  137.63  4601.2  135.95  4621.2  134.87
  4631.2  133.76  4711.2  129.15  4771.2  130.53  4790.6  130.13  4810.6  129.73
  4840.6  129.11  4841.2   129.1  4871.2   129.6  4881.2  129.32  4901.2  129.91
 4930.91  129.49    4931  129.49  4940.6  129.36  4951.2  129.21  4967.5  127.97
  4979.5  127.05  4986.5  122.25  5013.5  122.25  5020.5  127.05  5032.5  127.53
 5068.89  129.01    5069  129.01  5108.6  130.61  5128.6  131.13  5248.6  131.61
  5304.5  133.96  5314.5  134.39  5324.5  134.81  5334.5  135.23  5338.6   135.4
  5344.5  135.49  5374.5  135.96  5398.6  136.33  5424.5  139.02  5454.5  142.13
  5468.6  143.59  5488.6  147.59  5608.6  146.54  5794.5  149.29  5884.5  150.63
  5914.5  151.07  5964.5  151.81  6028.6  152.76  6034.5  152.95  6234.5  159.26
  6298.6  161.29  6327.2   161.6  6534.5  163.66  6564.5  163.95  6624.6  164.55
BR U #Mann= 3
 4135.30   0.131  4979.5   0.055  5020.5   0.131
BR U Banks=4979.50,5020.50
BR D #Sta/Elev= 75
  4135.3  162.38  4181.2   152.5  4201.2  151.39  4211.2  150.45  4225.3  149.98
  4241.2  149.45  4245.3  149.35  4265.3  148.83  4310.6  147.68  4311.2  147.66
  4321.2  146.96  4330.6  146.82  4331.2  146.81  4341.2  145.99  4371.2  145.86
  4381.2  144.73  4400.6  146.18  4401.2  146.22  4421.2  147.39  4431.2  147.17
  4441.2  146.14  4511.2  143.05  4580.6  137.38  4601.2   135.7  4621.2  134.62
  4631.2  133.51  4711.2   128.9  4771.2  130.28  4790.6  129.88  4810.6  129.48
  4840.6  128.86  4841.2  128.85  4871.2  129.35  4881.2  129.07  4901.2  129.66
 4930.91  129.24    4931  129.24  4940.6  129.11  4951.2  128.96  4967.5  127.72
  4979.5   126.8  4986.5     122  5013.5     122  5020.5   126.8  5032.5  127.28
 5068.89  128.76    5069  128.76  5108.6  130.36  5128.6  130.88  5248.6  131.36
  5304.5  133.71  5314.5  134.14  5324.5  134.56  5334.5  134.98  5338.6  135.15
  5344.5  135.24  5374.5  135.71  5398.6  136.08  5424.5  138.77  5454.5  141.88
  5468.6  143.34  5488.6  147.34  5608.6  146.29  5794.5  149.04  5884.5  150.38
  5914.5  150.82  5964.5  151.56  6028.6  152.51  6034.5   152.7  6234.5  159.01
  6298.6  161.04  6327.2  161.35  6534.5  163.41  6564.5   163.7  6624.6   164.3
BR D #Mann= 3
 4135.30   0.131  4979.5   0.055  5020.5   0.131
BR D Banks=4979.50,5020.50

Type RM Length L Ch R = 1 ,40183.9,392,392,392
BEGIN DESCRIPTION:
Downstream Section of Bridge/Culvert/Weir
END DESCRIPTION:
#Sta/Elev= 30
  4135.3  162.38  4181.2   152.5  4211.2  150.45  4311.2  147.66  4341.2  145.99
  4371.2  145.86  4381.2  144.73  4421.2  147.39  4431.2  147.17  4511.2  143.05
  4631.2  133.51  4711.2   128.9  4771.2  130.28  4841.2  128.85  4901.2  129.66
  4951.2  128.96  4979.5   126.8  4986.5     122  5013.5     122  5020.5   126.8
  5128.6  130.88  5248.6  131.36  5338.6  135.15  5398.6  136.08  5468.6  143.34
  5488.6  147.34  5608.6  146.29  6028.6  152.51  6298.6  161.04  6624.6   164.3
#Mann= 3 , 1 , 0
 4135.30   0.131       0  4979.5   0.055       0  5020.5   0.131       0
#XS Ineff= 2 , 0
       0    4920     136    5079       0     134
Bank Sta=4979.50,5020.50
Exp/Cntr=0.5,0.3

Type RM Length L Ch R = 1 ,39791.9,289.1,289.1,289.1
BEGIN DESCRIPTION:
Rocky Swamp 80.0
END DESCRIPTION:
#Sta/Elev= 30
  4288.5  152.38  4468.5  145.45  4688.5  139.23  4758.5  133.53  4858.5  130.57
  4878.5  128.12  4918.5  129.75  4958.5   129.5  4968.5  128.82  4983.7  124.95
  4985.2  121.95  5014.7  121.95  5016.2  124.95  5062.4  129.05  5112.4  131.57
  5132.4  131.54  5302.4  139.13  5402.4  137.24  5442.4  139.18  5502.4  139.99
  5552.4  138.86  5572.4  140.47  5652.4  142.24  5672.4  141.53  5812.4  144.36
  6042.4  145.78  6072.4  148.05  6342.4  153.16  6552.4  161.95  6564.2  163.34
#Mann= 3 , 1 , 0
 4288.50   0.131       0  4983.7   0.055       0  5016.2   0.131       0
Bank Sta=4983.70,5016.20
Exp/Cntr=0.3,0.1

Type RM Length L Ch R = 1 ,39502.8,502.8,502.8,502.8
BEGIN DESCRIPTION:
Rocky Swamp 79.0
END DESCRIPTION:
#Sta/Elev= 30
  4306.8  153.23  4326.8   151.4  4406.8  147.47  4436.8  144.67  4506.8  142.93
  4566.8  137.52  4646.8  134.54  4676.8  134.38  4716.8  131.16  4766.8  129.09
  4876.8  126.96  4916.8  127.41  4946.8  128.94  4983.8  124.92  4985.3  121.92
  5014.8  121.92  5016.3  124.92    5040  129.25    5140  129.25    5270  131.36
    5320  130.67    5380  134.71    5790  137.36    5860  139.03    5900  141.55
    6100  146.09    6550  150.43    6630  155.58    6660  159.93  6704.7  162.62
#Mann= 3 , 1 , 0
 4306.80   0.141       0  4983.8   0.055       0  5016.3   0.141       0
Bank Sta=4983.80,5016.30
Exp/Cntr=0.3,0.1

Type RM Length L Ch R = 1 ,39000.0,502,502,502
BEGIN DESCRIPTION:
Rocky Swamp 78.0
END DESCRIPTION:
#Sta/Elev= 30
  4372.6  154.33  4442.6  150.71  4532.6  143.69  4582.6  135.24  4622.6  130.77
  4952.6  129.38  4983.8  124.86  4985.3  121.86  5014.7  121.86  5016.2  124.86
    5040   130.7    5110  128.26    5230   130.1    5420  129.09    5530  132.06
    5550  130.88    5650  132.24    5690  131.38    5770  133.84    5940  135.23
    6130  139.85    6230  144.39    6260  143.52    6300  145.62    6330  144.64
    6430  147.59    6790  151.19    6880   154.9    6970  161.94  7059.9  165.37
#Mann= 3 , 1 , 0
 4372.60   0.141       0  4983.8   0.055       0  5016.2   0.141       0
Bank Sta=4983.80,5016.20
Exp/Cntr=0.3,0.1

Type RM Length L Ch R = 1 ,38498.0,500.3,500.3,500.3
BEGIN DESCRIPTION:
Rocky Swamp 77.0
END DESCRIPTION:
#Sta/Elev= 30
  4253.6  153.85  4393.6  148.33  4493.6  132.43  4553.6   129.5  4724.9  129.83
  4783.6  126.82  4873.6  129.79  4963.6  128.95  4973.6  128.55  4983.7  124.81
  4985.2  121.81  5014.7  121.81  5016.2  124.81    5030  128.84    5040  129.22
    5200  127.34  5324.9  128.82    5560  126.93    5610  128.26    6260  127.44
    6420  132.65    6780  131.01    6800  132.73    6880  133.04    6920  138.26
    6970  154.74    7080  173.01    7170   183.4    7240  188.85  7335.2  190.94
#Mann= 5 , 1 , 0
 4253.60       1       0  4724.9    0.15       0  4983.7   0.055       0
  5016.2    0.15       0  5324.9       1       0
Bank Sta=4983.70,5016.20
Exp/Cntr=0.3,0.1

Type RM Length L Ch R = 1 ,37997.7,501.8,501.8,501.8
BEGIN DESCRIPTION:
Rocky Swamp 76.0
END DESCRIPTION:
#Sta/Elev= 30
  3959.4  163.11  4119.4  158.83  4209.4  151.64  4249.4  146.89  4289.4  145.21
  4399.4  135.92  4479.4  127.77  4519.4  128.43  4549.4  126.32  4639.9  128.19
  4929.4  127.19  4949.4  128.57  4969.4  127.82  4983.7  124.75  4985.2  121.75
  5014.7  121.75  5016.2  124.75    5050  128.54  5330.9  127.01    5910   125.8
    6140  126.68    6400  129.97    6600   129.8    6660  134.06    6690   133.1
    6850  147.71    6980  153.92    7110  164.78    7240  179.07  7351.6  182.57
#Mann= 5 , 1 , 0
 3959.40       1       0  4639.9    0.15       0  4983.7   0.055       0
  5016.2    0.15       0  5330.9       1       0
Bank Sta=4983.70,5016.20
Exp/Cntr=0.3,0.1

Type RM Length L Ch R = 1 ,37495.9,499.3,499.3,499.3
BEGIN DESCRIPTION:
Rocky Swamp 75.0
END DESCRIPTION:
#Sta/Elev= 30
  3768.2  161.37  4048.2  154.49  4118.2  148.87  4178.2  146.33  4308.2  133.67
  4388.2  129.33  4538.2  127.49  4638.2  128.31  4678.2  126.41  4708.2  127.52
  4738.2  124.09  4769.9   127.5  4958.2  127.13  4983.8   124.7  4985.3   121.7
  5014.8   121.7  5016.3   124.7    5030  127.52    5240  125.86  5371.9  126.99
    5710  125.13    5820  126.81    5900  125.45    6450  127.11    6590  133.69
    6670  145.58    6760  151.81    6860   161.9    6920  164.49    7048  174.78
#Mann= 5 , 1 , 0
 3768.20       1       0  4769.9    0.15       0  4983.8   0.055       0
  5016.3    0.15       0  5371.9       1       0
Bank Sta=4983.80,5016.30
Exp/Cntr=0.3,0.1

Type RM Length L Ch R = 1 ,36996.6,584.2,584.2,584.2
BEGIN DESCRIPTION:
Rocky Swamp 74.0
END DESCRIPTION:
#Sta/Elev= 30
  4182.3  157.12  4242.3  155.19  4262.3  153.51  4282.3  150.28  4302.3  145.41
  4342.3  137.84  4392.3  130.22  4432.3  126.14  4452.3  125.02  4472.3  126.06
  4615.9  126.49  4902.3  124.33  4932.3  126.57  4983.8  124.64  4985.3  121.64
  5014.7  121.64  5016.2  124.64    5030  126.96    5050   125.6    5340  125.29
  5594.9  126.92    5620  124.73    5650  125.81    6100  126.14    6410  127.68
    6540  145.83    6580  149.36    6630  151.69    6740  162.26  6786.7  165.22
#Mann= 5 , 1 , 0
 4182.30       1       0  4615.9    0.15       0  4983.8   0.055       0
  5016.2    0.15       0  5594.9       1       0
Bank Sta=4983.80,5016.20
Exp/Cntr=0.3,0.1

Type RM Length L Ch R = 1 ,36412.4,548.5,548.5,548.5
BEGIN DESCRIPTION:
Rocky Swamp 73.0
END DESCRIPTION:
#Sta/Elev= 30
  4389.2  151.91  4479.2   145.9  4809.2  134.44  4869.2  129.42  4919.2  126.53
  4959.2  124.63  4983.8  124.58  4985.3  121.58  5014.7  121.58  5016.2  124.58
  5074.9  126.26  5134.9  127.06  5244.9  125.19  5273.9  125.37  5544.9  124.59
  5614.9  125.47  5714.9  125.21  5864.9  126.41  5944.9  126.41  5984.9  127.76
  6284.9  127.89  6334.9  126.75  6374.9  127.67  6384.9   127.3  6424.9  129.65
  6474.9  131.14  6534.9  136.04  6574.9  138.64  6644.9  149.93  6699.9  156.05
#Mann= 4 , 1 , 0
 4389.20   0.141       0  4983.8   0.055       0  5016.2   0.141       0
  5273.9       1       0
Bank Sta=4983.80,5016.20
Exp/Cntr=0.3,0.1

Type RM Length L Ch R = 1 ,35863.9,372,372,372
BEGIN DESCRIPTION:
Rocky Swamp 72.0
END DESCRIPTION:
#Sta/Elev= 30
  4064.8  154.46  4094.8  153.43  4174.8  144.85  4354.8  135.76  4514.8  133.81
  4644.8  128.19  4884.8  127.11  4982.6  124.53  4984.1  121.53  5015.8  121.53
  5017.3  124.53  5025.8  125.82  5055.8   124.7  5145.8  125.38  5175.8  124.73
  5195.8  125.85  5225.8  124.52  5275.8  125.85  5295.8  124.94  5525.8  124.96
  6175.8  126.47  6295.8  129.81  6325.8     132  6385.8  140.86  6395.8  143.69
  6415.8  146.68  6445.8  153.97  6495.8  159.39  6525.8  164.11  6546.7  165.24
#Mann= 3 , 1 , 0
 4064.80   0.141       0  4982.6   0.055       0  5017.3   0.141       0
Bank Sta=4982.60,5017.30
Exp/Cntr=0.3,0.1

Type RM Length L Ch R = 1 ,35491.9,500.2,500.2,500.2
BEGIN DESCRIPTION:
Rocky Swamp 71.0
END DESCRIPTION:
#Sta/Elev= 30
  3873.8   155.8  3903.8  153.72  3943.8   147.3  4013.8   142.1  4203.8  137.71
  4243.8  137.88  4413.8  131.25  4463.8  127.85  4773.8  124.67  4923.8   125.5
  4982.6  124.49  4984.1  121.49  5015.8  121.49  5017.3  124.49    5250  123.65
    5640  124.36    5660  125.22    5740  124.56    5900   126.3    6040  126.51
    6090  124.88    6250  127.33    6310  130.01    6370  141.18    6400  150.57
    6410   149.8    6450  157.37    6490  162.26    6510  165.76  6538.5     167
#Mann= 3 , 1 , 0
 3873.80   0.141       0  4982.6   0.055       0  5017.3   0.141       0
Bank Sta=4982.60,5017.30
Exp/Cntr=0.3,0.1

Type RM Length L Ch R = 1 ,34991.7,501.1,501.1,501.1
BEGIN DESCRIPTION:
Rocky Swamp 70.0
END DESCRIPTION:
#Sta/Elev= 30
  3651.4  156.16  3721.4  153.03  3791.4  144.21  3811.4  142.78  3951.4  136.92
  4121.4  133.61  4151.4  131.06  4311.4  126.03  4511.4  124.03  4561.4  125.14
  4921.4  125.23  4982.6  122.75  4984.1  119.75  5015.8  119.75  5017.3  122.75
    5070  124.76    5240  123.08    5510  124.11    5720   123.3    6040  125.57
    6070  124.36    6200  126.49    6340  126.32    6450  128.33    6460  129.07
    6530  140.75    6560  143.19    6580  147.41    6630  151.47  6668.4  156.19
#Mann= 3 , 1 , 0
 3651.40   0.141       0  4982.6   0.055       0  5017.3   0.141       0
Bank Sta=4982.60,5017.30
Exp/Cntr=0.3,0.1

Type RM Length L Ch R = 1 ,34490.6,498.9,498.9,498.9
BEGIN DESCRIPTION:
Rocky Swamp 69.0
END DESCRIPTION:
#Sta/Elev= 30
  3315.8   151.8  3405.8     150  3585.8  139.24  3745.8  135.14  3785.8  132.28
  3895.8  128.52  4105.8  125.49  4295.8  126.15  4355.8   124.8  4485.8  124.64
  4525.8  125.53  4735.8  123.85  4775.8  122.45  4905.8  124.32  4982.7  122.49
  4984.2  119.49  5015.8  119.49  5017.3  122.49    5040  124.32    5160  122.77
    5620  122.51    5630  124.57    5640  123.09    5660  122.46    6180  122.08
    6310  124.58    6350  132.36    6430   155.8    6500  172.54  6523.3  175.16
#Mann= 3 , 1 , 0
 3315.80   0.141       0  4982.7   0.055       0  5017.3   0.141       0
Bank Sta=4982.70,5017.30
Exp/Cntr=0.3,0.1

Type RM Length L Ch R = 1 ,33991.7,501.3,501.3,501.3
BEGIN DESCRIPTION:
Rocky Swamp 68.0
END DESCRIPTION:
#Sta/Elev= 30
  3004.4  151.26  3104.4  149.62  3214.4  143.71  3324.4  139.29  3444.4  137.06
  3634.4  131.79  3664.4  129.93  3794.4  128.25  4264.4  126.42  4294.4  127.54
  4584.9  129.91  4704.4  125.25  4864.4  124.86  4982.6  121.89  4984.1  118.89
  5015.8  118.89  5017.3  121.89    5040  124.23    5100  124.71    5150  123.03
    5470  122.15    5490  124.18    5510  122.01    5610  121.48    5650   122.8
    5980  123.72    6010  125.58    6090  143.79    6150  155.04  6182.7  158.55
#Mann= 4 , 1 , 0
 3004.40       1       0  4584.9   0.141       0  4982.6   0.055       0
  5017.3   0.141       0
Bank Sta=4982.60,5017.30
Exp/Cntr=0.3,0.1

Type RM Length L Ch R = 1 ,33490.4,499.5,499.5,499.5
BEGIN DESCRIPTION:
Rocky Swamp 67.0
END DESCRIPTION:
#Sta/Elev= 30
  2323.2  150.55  2613.2  149.39  2743.2   146.9  2823.2  143.69  3093.2  142.85
  3623.2  135.74  3923.2  133.58  4083.2  128.18  4123.2  128.34  4153.2  127.19
  4393.2  128.25  4423.2  127.41  4493.2  128.53  4633.2  126.61  4713.2  122.99
  4943.2  123.46  4982.7  121.59  4984.2  118.59  5015.8  118.59  5017.3  121.59
    5040  123.04    5550  121.45    5600  124.17    5620  122.32    5930   121.5
    5970  122.83    6110  122.45    6170  135.11    6230  145.33    6240  146.05
#Mann= 3 , 1 , 0
 2323.20   0.141       0  4982.7   0.055       0  5017.3   0.141       0
Bank Sta=4982.70,5017.30
Exp/Cntr=0.3,0.1

Type RM Length L Ch R = 1 ,32990.9,497.4,497.4,497.4
BEGIN DESCRIPTION:
Rocky Swamp 66.0
END DESCRIPTION:
#Sta/Elev= 30
  2166.2  153.01  2286.2  150.84  2396.2  147.08  2636.2  143.16  3286.2  141.87
  3396.2  138.09  3726.2  137.92  3866.2  134.22  4006.2  133.11  4146.2  129.26
  4346.2  126.28  4506.2  126.91  4616.2  124.47  4976.2  122.36  4982.6  121.33
  4984.1  118.33  5015.8  118.33  5017.3  121.33    5240  122.16    5350  119.92
    5370   121.5    5470  121.16    5560  124.42    5650  121.33    5730  122.23
    5750  123.67    5790  130.85    5850  144.41    5960  149.63  6021.1  150.62
#Mann= 3 , 1 , 0
 2166.20   0.141       0  4982.6   0.055       0  5017.3   0.141       0
Bank Sta=4982.60,5017.30
Exp/Cntr=0.3,0.1
