HEC-RAS study 020822_SANDY_CREEK.prj: Sandy Creek

--- 020822_SANDY_CREEK.g01 (geometry) --- (continued)

Type RM Length L Ch R = 1 ,241177.4,1172.1,1172.1,1172.1
BEGIN DESCRIPTION:
Sandy Creek 241.0
END DESCRIPTION:
#Sta/Elev= 30
  4646.6  392.35  4666.6  390.56  4676.6  390.54  4686.6  389.41  4706.6     385
  4816.6  370.67  4866.6  365.63  4886.6  364.85  4926.6  366.73  4986.6  366.75
  4990.4  364.98  4993.4  358.98  5006.6  358.98  5009.6  364.98  5018.5  366.46
  5118.5  365.56  5128.5  364.76  5138.5  364.67  5168.5  368.35  5198.5  369.79
  5238.5  369.42  5348.5  374.38  5378.5  377.09  5388.5  376.87  5408.5  377.82
  5508.5   388.7  5528.5  389.34  5558.5  393.92  5598.5  395.98  5616.7  396.22
#Mann= 3 , 1 , 0
 4646.60    0.13       0  4990.4   0.042       0  5009.6    0.13       0
Bank Sta=4990.40,5009.60
Exp/Cntr=0.3,0.1

Type RM Length L Ch R = 1 ,240005.3,1082.4,1082.4,1082.4
BEGIN DESCRIPTION:
Sandy Creek 240.0
END DESCRIPTION:
#Sta/Elev= 20
  4803.4  392.96  4823.4  390.99  4933.4     372  4943.4  369.52  4973.4  364.45
  4990.4  364.13  4993.4  358.13  5006.6  358.13  5009.6  364.13  5043.7  364.18
  5063.7  365.42  5073.7  365.05  5083.7  365.46  5113.7  368.31  5133.7  371.32
  5233.7  382.19  5293.7  387.24  5363.7  395.54  5433.7  399.18  5448.7  399.23
#Mann= 3 , 1 , 0
 4803.40    0.13       0  4990.4   0.042       0  5009.6    0.13       0
Bank Sta=4990.40,5009.60
Exp/Cntr=0.3,0.1

Type RM Length L Ch R = 1 ,238922.9,1002.7,1002.7,1002.7
BEGIN DESCRIPTION:
Sandy Creek 239.0
END DESCRIPTION:
#Sta/Elev= 30
  4430.3  392.08  4460.3  389.89  4500.3  388.35  4520.3  386.17  4580.3  382.26
  4600.3  380.35  4690.3   375.3  4750.3  371.72  4770.3   371.2  4790.3  369.63
  4800.3  369.61  4840.3  367.53  4860.3  367.07  4870.3  367.68  4890.3  367.17
  4900.3  366.29  4930.3  365.26  4960.3   365.2  4970.3  363.07  4990.4  362.81
  4993.4  356.81  5006.7  356.81  5009.7  362.81    5060  362.92    5070  368.17
    5080  374.93    5100  389.96    5110  395.34    5120  399.39  5130.2  402.43
#Mann= 3 , 1 , 0
 4430.30    0.13       0  4990.4   0.042       0  5009.7    0.13       0
Bank Sta=4990.40,5009.70
Exp/Cntr=0.3,0.1

Type RM Length L Ch R = 1 ,237920.2,998.3,998.3,998.3
BEGIN DESCRIPTION:
Sandy Creek 237.5
END DESCRIPTION:
#Sta/Elev= 17
  4669.5   398.2  4709.5  395.87  4739.5  393.06  4749.5  392.48  4799.5  385.46
  4879.5  369.76  4990.4   359.6  4993.4   353.6  5006.6   353.6  5009.6   359.6
  5036.4  359.23  5076.4  369.12  5086.4  370.48  5186.4  376.45  5246.4   383.9
  5276.4  386.29  5327.5  391.54
#Mann= 3 , 1 , 0
 4669.50    0.13       0  4990.4   0.042       0  5009.6    0.13       0
Bank Sta=4990.40,5009.60
Exp/Cntr=0.3,0.1

Type RM Length L Ch R = 1 ,236921.9,1121.8,1121.8,1121.8
BEGIN DESCRIPTION:
Sandy Creek 237.0
END DESCRIPTION:
#Sta/Elev= 30
  4639.7  375.81  4669.7  374.28  4699.7  373.83  4719.7  371.44  4759.7   363.7
  4769.7  362.13  4779.7  361.64  4789.7  361.75  4799.7  361.08  4809.7  361.08
  4819.7  359.72  4839.7  355.48  4869.7  351.48  4909.7  351.42  4919.7   352.5
  4929.7  352.85  4939.7  351.59  4949.7  349.61  4959.7  350.13  4990.4  348.31
  4993.4  342.31  5006.6  342.31  5009.6  348.31    5010  366.91    5020  376.88
    5030  383.21    5040  388.89    5050  395.65    5060  399.95  5065.6  401.13
#Mann= 3 , 1 , 0
 4639.70    0.13       0  4990.4   0.042       0  5009.6    0.13       0
Bank Sta=4990.40,5009.60
Exp/Cntr=0.3,0.1

Type RM Length L Ch R = 1 ,235800.1,979.1,979.1,979.1
BEGIN DESCRIPTION:
Sandy Creek 236.0
END DESCRIPTION:
#Sta/Elev= 29
  4578.7  375.76  4658.7  370.19  4678.7  368.27  4708.7  365.92  4728.7  362.87
  4738.7  362.23  4778.7  356.37  4788.7  354.34  4808.7  348.03  4818.7  345.82
  4838.7  342.63  4848.7  341.57  4868.7  341.12  4928.7  343.45  4989.2  341.08
  4992.2  335.08  5007.8  335.08  5010.8  341.08  5016.8   347.6  5026.8   349.4
  5076.8  353.24  5086.8  354.88  5096.8  355.74  5106.8  357.41  5156.8  362.67
  5176.8  365.76  5246.8  371.06  5266.8  373.13  5273.9  373.32
#Mann= 3 , 1 , 0
 4578.70    0.13       0  4989.2   0.042       0  5010.8    0.13       0
Bank Sta=4989.20,5010.80
Exp/Cntr=0.3,0.1

Type RM Length L Ch R = 1 ,234821.0,1140.5,1140.5,1140.5
BEGIN DESCRIPTION:
Sandy Creek 235.0
END DESCRIPTION:
#Sta/Elev= 20
  4555.7  369.89  4613.1  365.61  4623.1  365.63  4783.1  352.91  4853.1  344.24
  4863.1   343.7  4913.1  345.16  4933.1  344.88  4953.1  343.45  4956.8  343.17
  4986.8  340.03  4989.2  338.55  4992.2  332.55  5007.9  332.55  5010.9  338.55
  5016.8  348.34  5026.8  352.53  5036.8  356.18  5066.8  361.67  5086.8  366.55
#Mann= 3 , 1 , 0
 4555.70    0.13       0  4989.2   0.042       0  5010.9    0.13       0
Bank Sta=4989.20,5010.90
Exp/Cntr=0.3,0.1

Type RM Length L Ch R = 1 ,233680.5,1171.4,1171.4,1171.4
BEGIN DESCRIPTION:
Sandy Creek 234.0
END DESCRIPTION:
#Sta/Elev= 16
  4708.5  364.08  4728.5  363.18  4838.5  354.58  4848.5  353.34  4928.5  339.59
  4989.2  336.89  4992.2  330.89  5007.8  330.89  5010.8  336.89  5086.4  336.93
  5126.4  338.99  5256.4  344.66  5286.4   346.9  5306.4  351.39  5366.4  358.45
  5436.5  364.35
#Mann= 3 , 1 , 0
 4708.50    0.13       0  4989.2   0.042       0  5010.8    0.13       0
Bank Sta=4989.20,5010.80
Exp/Cntr=0.3,0.1

Type RM Length L Ch R = 1 ,232509.1,1593.7,1593.7,1593.7
BEGIN DESCRIPTION:
Sandy Creek 233.0
END DESCRIPTION:
#Sta/Elev= 14
  4578.9  367.25  4608.9  367.07  4638.9  365.34  4678.9  361.52  4728.9   353.1
  4798.9  339.47  4986.1  334.76  4989.1  328.76    5011  328.76    5014  334.76
  5173.2     336  5273.2  349.07  5303.2  356.92  5372.7  369.05
#Mann= 3 , 1 , 0
 4578.90    0.13       0  4986.1   0.042       0    5014    0.13       0
Bank Sta=4986.10,5014.00
Exp/Cntr=0.3,0.1

Type RM Length L Ch R = 1 ,230915.4,832.6,832.6,832.6
BEGIN DESCRIPTION:
Sandy Creek 232.0
END DESCRIPTION:
#Sta/Elev= 30
    4281  354.41    4351  351.85    4381  352.23    4391  353.08    4421  353.73
    4441  353.44    4481   353.9    4491  354.79    4511  354.82    4521  355.74
    4531  355.24    4561  355.49    4591  357.75    4661  355.23    4711   354.1
    4731  352.17    4741  351.83    4851  340.87    4891  338.59    4911  338.14
    4986  332.71    4989  326.71  5010.9  326.71  5013.9  332.71  5068.8  335.26
  5088.8  337.37  5338.8  337.08  5388.8  340.39  5468.8  355.91  5510.4  358.96
#Mann= 3 , 1 , 0
 4281.00    0.13       0    4986   0.042       0  5013.9    0.13       0
Bank Sta=4986.00,5013.90
Exp/Cntr=0.3,0.1

Type RM Length L Ch R = 1 ,230082.8,734.5,734.5,734.5
BEGIN DESCRIPTION:
Sandy Creek 231.0
END DESCRIPTION:
#Sta/Elev= 27
  4246.3   360.7  4276.3  359.08  4286.3     358  4296.3  357.66  4326.3  354.66
  4406.3  350.62  4416.3   350.4  4456.3  347.21  4499.9  341.67  4556.3  334.51
  4566.3  334.22  4606.3  335.98  4636.3  336.82  4766.3  336.13  4796.3  336.69
  4836.3   334.8  4856.3  336.84  4926.3  335.26  4966.3  336.34  4976.3  334.56
  4984.8  333.92  4986.1  332.09  4989.1  326.09    5011  326.09    5014  332.09
  5034.8  361.12  5064.7  368.71
#Mann= 4 , 1 , 0
 4246.30       1       0  4499.9    0.13       0  4986.1   0.042       0
    5014    0.13       0
Bank Sta=4986.10,5014.00
Exp/Cntr=0.3,0.1

Type RM Length L Ch R = 1 ,229348.3,604.9,604.9,604.9
BEGIN DESCRIPTION:
Sandy Creek 230.0
END DESCRIPTION:
#Sta/Elev= 30
  4002.2  369.43  4062.2  364.22  4072.2   362.9  4092.2   358.8  4112.2  352.46
  4152.2  341.09  4162.2   338.9  4172.2  338.07  4202.2  337.01  4232.2  334.48
  4462.2  334.62  4499.9  333.88  4592.2   334.6  4622.2  334.33  4642.2  335.18
  4942.2   335.6  4952.2  336.34  4971.6  334.25  4981.6  335.19  4986.1  328.24
  4989.1  322.24    5011  322.24    5014  328.24  5021.6  336.32  5041.6  337.95
  5051.6  339.55  5071.6  344.59  5091.6  351.11  5121.6  356.65  5168.6  361.63
#Mann= 4 , 1 , 0
 4002.20       1       0  4499.9    0.13       0  4986.1   0.042       0
    5014    0.13       0
Bank Sta=4986.10,5014.00
Exp/Cntr=0.3,0.1

Type RM Length L Ch R = 1 ,228743.4,809.1,809.1,809.1
BEGIN DESCRIPTION:
Sandy Creek 229.0
END DESCRIPTION:
#Sta/Elev= 30
  4570.8  362.51  4580.8  360.95  4610.8  359.52  4660.8  355.69  4720.8  348.67
  4740.8  347.12  4810.8  337.45  4820.8  335.29  4830.8  333.67  4840.8   332.7
  4880.8  331.68  4920.8  332.26  4940.8  330.75  4950.8  331.16  4960.8  330.13
  4970.8  328.45  4986.1  328.24  4989.1  322.24  5010.9  322.24  5013.9  328.24
  5016.6  333.78  5036.6  333.42  5046.6  333.69  5066.6   337.1  5076.6  338.21
  5096.6   342.5  5136.6  349.17  5156.6  353.13  5246.6  361.33  5251.4  361.43
#Mann= 3 , 1 , 0
 4570.80    0.13       0  4986.1   0.042       0  5013.9    0.13       0
Bank Sta=4986.10,5013.90
Exp/Cntr=0.3,0.1

Type RM Length L Ch R = 1 ,227934.3,771.3,771.3,771.3
BEGIN DESCRIPTION:
Sandy Creek 228.0
END DESCRIPTION:
#Sta/Elev= 27
  4729.2  355.99  4759.2  352.18  4829.2  344.37  4849.2  342.97  4869.2  340.79
  4879.2  339.25  4899.2   337.3  4909.2  335.73  4929.2  331.59  4949.2  330.11
  4986.1  328.01  4989.1  322.01    5011  322.01    5014  328.01  5029.3  334.14
  5059.3  336.88  5079.3   339.9  5089.3  340.77  5119.3  341.03  5189.3  345.79
  5219.3  348.13  5239.3  348.49  5249.3  350.43  5309.3  355.55  5349.3  357.88
  5379.3  358.85  5418.9  361.95
#Mann= 3 , 1 , 0
 4729.20    0.13       0  4986.1   0.042       0    5014    0.13       0
Bank Sta=4986.10,5014.00
Exp/Cntr=0.3,0.1

Type RM Length L Ch R = 1 ,227163.0,639,639,639
BEGIN DESCRIPTION:
Sandy Creek 227.0
END DESCRIPTION:
#Sta/Elev= 28
    4705  366.82    4755  359.95    4795   354.9    4805  353.31    4845  342.97
    4865  340.35    4895  335.06    4915  329.63    4955  325.99    4985  327.82
    4986  324.49    4989  318.49  5010.9  318.49  5013.9  324.49  5018.6  330.89
  5028.6  333.83  5038.6   336.1  5048.6   337.4  5068.6  342.56  5088.6   345.6
  5098.6  346.64  5118.6   350.1  5198.6  360.99  5228.6  364.32  5248.6  366.05
  5268.6  368.83  5288.6  369.58  5292.2  369.87
#Mann= 3 , 1 , 0
 4705.00    0.13       0    4986   0.042       0  5013.9    0.13       0
Bank Sta=4986.00,5013.90
Exp/Cntr=0.3,0.1

Type RM Length L Ch R = 1 ,226524.0,773.2,773.2,773.2
BEGIN DESCRIPTION:
Sandy Creek 226.0
END DESCRIPTION:
#Sta/Elev= 27
  4592.3  363.05  4652.3  356.96  4772.3  343.26  4792.3  340.12  4812.3  336.17
  4822.3  334.88  4832.3  332.93  4842.3  330.26  4852.3  326.79  4862.3  324.97
  4872.3   324.7  4942.3  324.44  4986.1  322.26  4989.1  316.26    5011  316.26
    5014  322.26  5027.7   326.1  5037.7  328.52  5047.7  334.12  5057.7   338.2
  5087.7   347.1  5107.7  351.21  5147.7  357.49  5197.7  363.67  5267.7  369.88
  5277.7   371.2  5292.2  372.31
#Mann= 3 , 1 , 0
 4592.30    0.13       0  4986.1   0.042       0    5014    0.13       0
Bank Sta=4986.10,5014.00
Exp/Cntr=0.3,0.1

Type RM Length L Ch R = 1 ,225750.8,1702,1702,1702
BEGIN DESCRIPTION:
Sandy Creek 225.0
END DESCRIPTION:
#Sta/Elev= 18
  4330.4  351.59  4440.4  341.21  4590.4  321.89  4760.4  321.92  4970.4  324.02
  4986.1  321.75  4989.1  315.75    5011  315.75    5014  321.75    5022  324.02
    5062  323.34    5082  326.17    5172  346.73    5182  348.28    5292  358.84
    5312  359.77    5322  359.69  5404.2  363.91
#Mann= 3 , 1 , 0
 4330.40    0.13       0  4986.1   0.042       0    5014    0.13       0
Bank Sta=4986.10,5014.00
Exp/Cntr=0.3,0.1

Type RM Length L Ch R = 1 ,224048.8,1425.5,1425.5,1425.5
BEGIN DESCRIPTION:
Sandy Creek 224.0
END DESCRIPTION:
#Sta/Elev= 15
  4622.1  351.69  4672.1  346.15  4822.1  323.06  4832.1  321.81  4912.1  320.78
  4984.3  320.51  4987.3  314.51  5012.6  314.51  5015.6  320.51  5043.1  333.56
  5063.1  340.42  5073.1  342.71  5103.1  346.51  5123.1  348.35  5128.7  349.22
#Mann= 3 , 1 , 0
 4622.10    0.13       0  4984.3   0.042       0  5015.6    0.13       0
Bank Sta=4984.30,5015.60
Exp/Cntr=0.3,0.1

Type RM Length L Ch R = 1 ,222623.3,22,22,22
BEGIN DESCRIPTION:
Upstream Section of Bridge/Culvert/Weir
END DESCRIPTION:
#Sta/Elev= 24
  4754.6  336.91  4774.6  333.85  4784.6  331.03  4794.6  330.54  4804.6  328.96
  4814.6  326.38  4834.6  324.94  4865.6   325.1  4884.6   325.2  4944.6  323.83
  4954.6  323.02    4974  314.16  4999.9  311.16  5000.1  311.16    5026  314.16
  5085.7  323.53  5095.7  323.03  5105.7  325.39  5115.7  327.18  5175.7  331.09
  5204.6  332.29  5285.7  335.65  5335.7  337.04  5345.7   337.8
#Mann= 3 , 1 , 0
 4754.60    0.13       0    4974   0.045       0    5026    0.13       0
#XS Ineff= 2 , 0
       0    4964  320.24    5036       0  320.24
Bank Sta=4974.00,5026.00
Exp/Cntr=0.5,0.3

Type RM Length L Ch R = 5 ,222612.3,,,
BEGIN DESCRIPTION:
Dam_Weldon Mill Rd_2
Structure ID: Dam_weldon Mill Rd
Approximate Survey Structure
END DESCRIPTION:
#Inline Weir SE= 24
  4754.6  334.02  4774.6  330.96  4784.6  328.14  4794.6  327.65  4804.6  326.07
  4814.6  323.49  4834.6  322.05  4865.6  322.22  4884.6  322.32  4944.6  320.95
  4954.6  320.14    4974     320  4999.9     320  5000.1     320    5026     320
  5085.7  320.65  5095.7  320.15  5105.7  322.51  5115.7   324.3  5175.7  328.21
  5204.6  329.41  5285.7  332.76  5335.7  334.15  5345.7  334.91
IW Dist,WD,Coef,Skew,MaxSub,Min_El,Is_Ogee,SpillHt,DesHd
10.0,2.0,3.0,,0.95,, 0 ,,,2.0,2.0,

Type RM Length L Ch R = 1 ,222601.3,163.4,163.4,163.4
BEGIN DESCRIPTION:
Downstream Section of Bridge/Culvert/Weir
END DESCRIPTION:
#Sta/Elev= 24
  4754.6  331.13  4774.6  328.07  4784.6  325.25  4794.6  324.76  4804.6  323.18
  4814.6   320.6  4834.6  319.16  4865.6  319.32  4884.6  319.42  4944.6  318.05
  4954.6  317.24    4974  308.38  4999.9  305.38  5000.1  305.38    5026  308.38
  5085.7  317.75  5095.7  317.25  5105.7  319.61  5115.7   321.4  5175.7  325.31
  5204.6  326.51  5285.7  329.87  5335.7  331.26  5345.7  332.02
#Mann= 3 , 1 , 0
 4754.60    0.13       0    4974   0.045       0    5026    0.13       0
#XS Ineff= 2 , 0
       0    4964  316.24    5036       0  316.24
Bank Sta=4974.00,5026.00
Exp/Cntr=0.5,0.3

Type RM Length L Ch R = 1 ,222437.9,45,45,45
BEGIN DESCRIPTION:
Upstream Section of Bridge/Culvert/Weir
END DESCRIPTION:
#Sta/Elev= 27
    4746  330.23    4756  328.75    4766  328.23    4776  328.95    4796   327.6
    4886  319.77    4906  318.43    4926  315.38    4946  315.02    4956  315.83
  4964.5  309.63    4978  303.63    5022  303.63  5035.5  309.63  5055.5  312.98
  5095.5  315.53  5105.5  315.81  5125.5  315.48  5165.5  316.89  5185.5  318.28
  5195.5  320.01  5205.5  322.31  5235.5  325.57  5245.5  326.15  5255.5  326.22
  5295.5  329.26  5385.4  329.46
#Mann= 3 , 1 , 0
 4746.00    0.13       0  4964.5   0.045       0  5035.5    0.13       0
#XS Ineff= 2 , 0
       0    4948  320.04    5051       0  320.39
Bank Sta=4964.50,5035.50
Exp/Cntr=0.5,0.3

Type RM Length L Ch R = 3 ,222415.4,,,
BEGIN DESCRIPTION:
Weldon Mill Rd-1-TOR
Structure ID: Weldon Mill Rd-Bridge
Approximate Survey Structure
END DESCRIPTION:
Bridge Culvert--1,0,-1,-1, 0
Deck Dist Width WeirC Skew NumUp NumDn MinLoCord MaxHiCord MaxSubmerge Is_Ogee
10,25,2.6,,42,42,,,0.95,0,1,1,,
    4746    4756    4766  4772.8    4776    4796  4812.8  4822.8  4852.8    4886
    4906    4926  4932.8    4946    4956 4959.41  4959.5    4961  4964.5    4978
    5022  5035.5    5039 5040.39  5040.5  5055.5  5095.5  5105.5  5125.5  5165.5
  5185.5  5195.5  5205.5  5235.5  5245.5  5255.5  5265.4  5295.5  5305.4  5325.4
  5375.4  5385.4
     331  329.52     329  331.84  331.33  328.38  326.92  326.05  323.44  322.02
  321.17  320.31  320.02  320.06  320.09   320.1   320.1   320.1  320.11  320.15
  320.27  320.31  320.32  320.33  320.33  320.37  320.48  320.51  320.57  320.68
  320.74  320.79  323.09  326.35  326.93     327  327.75  330.04  330.06  330.11
  330.22  330.23
  330.57  329.09  328.57  329.06  329.29  327.94  326.48  325.61     323  320.11
  318.77  315.72   315.6  315.36  316.17  313.68  317.07  317.07  317.08  317.12
  317.24  317.28  317.29   317.3  310.81  313.32  315.87  316.15  315.82  317.23
  318.62  320.35  322.65  325.91  326.49  326.56  327.31   329.6  329.62  329.67
  329.78   329.8
    4746    4756    4766  4772.8    4776    4796  4812.8  4822.8  4852.8    4886
    4906    4926  4932.8    4946    4956 4959.41  4959.5    4961  4964.5    4978
    5022  5035.5    5039 5040.39  5040.5  5055.5  5095.5  5105.5  5125.5  5165.5
  5185.5  5195.5  5205.5  5235.5  5245.5  5255.5  5265.4  5295.5  5305.4  5325.4
  5375.4  5385.4
  331.43  329.95  329.43  331.84  331.33   328.8  327.34  326.47  323.86  322.02
  321.17  320.31  320.02  320.06  320.09   320.1   320.1   320.1  320.11  320.15
  320.27  320.31  320.32  320.33  320.33  320.37  320.48  320.51  320.57  320.68
  320.74  321.21  323.51  326.77  327.35  327.42  328.17  330.46  330.48  330.53
  330.64  330.66
  331.43  329.95  329.43  329.92  330.15   328.8  327.34  326.47  323.86  320.97
  319.63  316.58  316.46  316.22  317.03  314.54  317.93  317.93  317.94  317.98
   318.1  318.14  318.15  318.16  311.67  314.18  316.73  317.01  316.68  318.09
  319.48  321.21  323.51  326.77  327.35  327.42  328.17  330.46  330.48  330.53
  330.64  330.66
Pier Skew, UpSta & Num, DnSta & Num=,5000.0, 2 ,5000.0, 2 , 0 , 0 , 0 ,,
       1       1
  302.97  318.18
       1       1
  303.83  319.04
Abutment Skew #Up #Dn=, 2 , 2
 4959.30 4961.00
  317.07  312.52
 4959.30 4961.00
  317.93  313.38
Abutment Skew #Up #Dn=, 2 , 2
 5039.00 5040.59
  310.56  317.30
 5039.00 5040.59
  311.42  318.16
BR Coef= 1 , 1 , 0 ,1.25, 0 ,,,0.8,0,2,0,
Wspro=,,,, 1 ,,,, 0 ,,,, 0 ,,,,-1 ,-1 ,-1 , 0 , 0 , 0 , 0 , 0
BC Design=,, 0 ,, 0 ,,,,,,
BR U #Sta/Elev= 42
    4746  330.57    4756  329.09    4766  328.57  4772.8  329.06    4776  329.29
    4796  327.94  4812.8  326.48  4822.8  325.61  4852.8     323    4886  320.11
    4906  318.77    4926  315.72  4932.8   315.6    4946  315.36    4956  316.17
 4959.41  313.68  4959.5  313.62    4961  312.52  4964.5  309.97    4978  303.97
    5022  303.97  5035.5  309.97    5039  310.56 5040.39  310.79  5040.5  310.81
  5055.5  313.32  5095.5  315.87  5105.5  316.15  5125.5  315.82  5165.5  317.23
  5185.5  318.62  5195.5  320.35  5205.5  322.65  5235.5  325.91  5245.5  326.49
  5255.5  326.56  5265.4  327.31  5295.5   329.6  5305.4  329.62  5325.4  329.67
  5375.4  329.78  5385.4   329.8
BR U #Mann= 3
 4746.00    0.13  4964.5   0.045  5035.5    0.13
BR U Banks=4964.50,5035.50
BR D #Sta/Elev= 42
    4746  331.43    4756  329.95    4766  329.43  4772.8  329.92    4776  330.15
    4796   328.8  4812.8  327.34  4822.8  326.47  4852.8  323.86    4886  320.97
    4906  319.63    4926  316.58  4932.8  316.46    4946  316.22    4956  317.03
 4959.41  314.54  4959.5  314.48    4961  313.38  4964.5  310.83    4978  304.83
    5022  304.83  5035.5  310.83    5039  311.42 5040.39  311.65  5040.5  311.67
  5055.5  314.18  5095.5  316.73  5105.5  317.01  5125.5  316.68  5165.5  318.09
  5185.5  319.48  5195.5  321.21  5205.5  323.51  5235.5  326.77  5245.5  327.35
  5255.5  327.42  5265.4  328.17  5295.5  330.46  5305.4  330.48  5325.4  330.53
  5375.4  330.64  5385.4  330.66
BR D #Mann= 3
 4746.00    0.13  4964.5   0.045  5035.5    0.13
BR D Banks=4964.50,5035.50

Type RM Length L Ch R = 1 ,222392.9,2003.4,2003.4,2003.4
BEGIN DESCRIPTION:
Downstream Section of Bridge/Culvert/Weir
END DESCRIPTION:
#Sta/Elev= 27
    4746  331.77    4756  330.29    4766  329.77    4776  330.49    4796  329.14
    4886  321.31    4906  319.97    4926  316.92    4946  316.56    4956  317.37
  4964.5  311.17    4978  305.17    5022  305.17  5035.5  311.17  5055.5  314.52
  5095.5  317.07  5105.5  317.35  5125.5  317.02  5165.5  318.43  5185.5  319.82
  5195.5  321.55  5205.5  323.85  5235.5  327.11  5245.5  327.69  5255.5  327.76
  5295.5   330.8  5385.4     331
#Mann= 3 , 1 , 0
 4746.00    0.13       0  4964.5   0.045       0  5035.5    0.13       0
#XS Ineff= 2 , 0
       0    4948  320.04    5051       0  320.39
Bank Sta=4964.50,5035.50
Exp/Cntr=0.5,0.3

Type RM Length L Ch R = 1 ,220389.5,528.5,528.5,528.5
BEGIN DESCRIPTION:
Sandy Creek 221.0
END DESCRIPTION:
#Sta/Elev= 22
  4599.6   334.7  4619.6  333.08  4719.6  328.37  4789.6  321.42  4829.6  315.38
  4859.6  308.11  4899.6  307.08  4959.6  307.12  4969.4  307.48  4979.4  307.78
  4981.5  308.05  4984.5  302.05  5015.4  302.05  5018.4  308.05  5119.4  307.21
  5339.4  308.17  5349.4  309.08  5369.4  312.37  5379.4  312.31  5409.4  320.21
  5439.4  325.69  5453.9  328.96
#Mann= 3 , 1 , 0
 4599.60    0.13       0  4981.5   0.042       0  5018.4    0.13       0
Bank Sta=4981.50,5018.40
Exp/Cntr=0.3,0.1

Type RM Length L Ch R = 1 ,219861.0,1022.7,1022.7,1022.7
BEGIN DESCRIPTION:
Sandy Creek 220.0
END DESCRIPTION:
#Sta/Elev= 21
  4646.1  334.68  4676.1   333.3  4736.1   327.9  4836.1  319.41  4856.1   315.8
  4886.1  309.21  4896.1  307.92  4956.1  306.68  4976.1  306.96  4981.6  305.95
  4984.6  299.95  5015.5  299.95  5018.5  305.95  5035.9  307.15  5195.9  307.44
  5505.9  306.59  5555.9   309.6  5565.9   313.1  5605.9  323.27  5675.9  332.53
  5684.7  333.26
#Mann= 3 , 1 , 0
 4646.10    0.13       0  4981.6   0.042       0  5018.5    0.13       0
Bank Sta=4981.60,5018.50
Exp/Cntr=0.3,0.1

Type RM Length L Ch R = 1 ,218838.3,711.5,711.5,711.5
BEGIN DESCRIPTION:
Sandy Creek 219.0
END DESCRIPTION:
#Sta/Elev= 23
  4724.6  334.56  4744.6  331.26  4774.6  323.08  4784.6  319.93  4804.6  312.69
  4814.6  309.57  4824.6  307.37  4834.6  306.05  4864.6  306.05  4874.6  305.61
  4981.6  305.07  4984.6  299.07  5015.5  299.07  5018.5  305.07  5062.4  305.44
  5092.4  305.66  5132.4  309.24  5152.4  309.16  5162.4   309.5  5212.4   320.2
  5242.4  325.01  5262.4  329.01  5285.6  332.08
#Mann= 3 , 1 , 0
 4724.60    0.13       0  4981.6   0.042       0  5018.5    0.13       0
Bank Sta=4981.60,5018.50
Exp/Cntr=0.3,0.1

Type RM Length L Ch R = 1 ,218126.8,1008.4,1008.4,1008.4
BEGIN DESCRIPTION:
Sandy Creek 218.0
END DESCRIPTION:
#Sta/Elev= 15
  4595.3  328.82  4635.3  325.41  4725.3  319.86  4795.3  311.44  4895.3  304.32
  4981.6  304.86  4984.6  298.86  5015.5  298.86  5018.5  304.86    5060  303.69
    5070  304.05    5080  307.23    5090  309.82    5130   335.5  5133.2  337.39
#Mann= 3 , 1 , 0
 4595.30    0.13       0  4981.6   0.042       0  5018.5    0.13       0
Bank Sta=4981.60,5018.50
Exp/Cntr=0.3,0.1

Type RM Length L Ch R = 1 ,217118.4,1119.3,1119.3,1119.3
BEGIN DESCRIPTION:
Sandy Creek 217.0
END DESCRIPTION:
#Sta/Elev= 20
  4757.2  331.73  4797.2  327.74  4857.2  322.18  4867.2  320.53  4917.2  308.15
  4927.2  306.46  4967.2  303.67  4981.5  304.59  4984.5  298.59  5015.4  298.59
  5018.4  304.59  5035.3  303.99  5045.3  305.04  5075.3  311.31  5095.3  314.99
  5125.3  319.66  5135.3  322.05  5205.3  332.26  5245.3  336.12  5247.2  336.25
#Mann= 3 , 1 , 0
 4757.20    0.13       0  4981.5   0.042       0  5018.4    0.13       0
Bank Sta=4981.50,5018.40
Exp/Cntr=0.3,0.1

Type RM Length L Ch R = 1 ,215999.1,1006,1006,1006
BEGIN DESCRIPTION:
Sandy Creek 216.0
END DESCRIPTION:
#Sta/Elev= 30
    4221   344.9    4311  337.74    4351  332.86    4371  327.83    4401  324.45
    4421  317.82    4481   301.5  4499.9  300.39    4531   300.2    4571  301.74
    4611  300.89    4691  305.24    4921  306.53    4981  304.31  4981.5   300.3
  4984.5   294.3  5015.4   294.3  5018.4   300.3    5020  302.02    5060  301.83
    5100  303.24    5150  303.28    5250  300.95    5280  302.66    5290  304.67
    5300  309.34    5310  315.94    5320  317.14    5340  324.46  5402.2  336.96
#Mann= 4 , 1 , 0
 4221.00       1       0  4499.9    0.13       0  4981.5   0.042       0
  5018.4    0.13       0
Bank Sta=4981.50,5018.40
Exp/Cntr=0.3,0.1

Type RM Length L Ch R = 1 ,214993.1,1360.2,1360.2,1360.2
BEGIN DESCRIPTION:
Sandy Creek 215.0
END DESCRIPTION:
#Sta/Elev= 30
  4701.2  338.68  4721.2   338.4  4741.2  337.12  4791.2  331.43  4831.2  324.92
  4871.2  312.55  4881.2  310.32  4901.2  304.17  4921.2  300.92  4981.5  300.09
  4984.5  294.09  5015.4  294.09  5018.4  300.09  5025.7  300.79  5055.7  301.52
  5065.7  301.03  5085.7   301.8  5115.7  306.39  5145.7   308.4  5175.7   309.5
  5205.7  312.94  5235.7  317.28  5265.7  319.53  5275.7  320.92  5285.7  321.01
  5305.7  323.32  5335.7  324.88  5345.7  324.71  5385.7   327.2  5480.3   328.6
#Mann= 3 , 1 , 0
 4701.20    0.13       0  4981.5   0.042       0  5018.4    0.13       0
Bank Sta=4981.50,5018.40
Exp/Cntr=0.3,0.1

Type RM Length L Ch R = 1 ,213632.9,842.7,842.7,842.7
BEGIN DESCRIPTION:
Sandy Creek 214.0
END DESCRIPTION:
#Sta/Elev= 17
  4721.7  331.68  4771.7  328.76  4851.7  320.05  4861.7   318.6  4891.7  312.86
  4941.7  305.11  4981.6  299.92  4984.6  293.92  5015.5  293.92  5018.5  299.92
  5030.8  301.05  5250.8  301.24  5330.8  308.27  5440.8  314.85  5500.8  319.82
  5540.8  321.23  5578.8  321.75
#Mann= 3 , 1 , 0
 4721.70    0.13       0  4981.6   0.042       0  5018.5    0.13       0
Bank Sta=4981.60,5018.50
Exp/Cntr=0.3,0.1

Type RM Length L Ch R = 1 ,212790.2,952.5,952.5,952.5
BEGIN DESCRIPTION:
Sandy Creek 213.0
END DESCRIPTION:
#Sta/Elev= 22
  4669.8  330.94  4759.8  323.11  4819.8  315.75  4859.8  308.07  4869.8  307.15
  4889.8  303.61  4929.8  301.05  4939.8  299.92  4981.6  299.82  4984.6  293.82
  5015.5  293.82  5018.5  299.82  5057.4  299.91  5087.4  301.51  5097.4  301.35
  5117.4  303.37  5147.4  307.97  5207.4  315.32  5237.4  317.27  5357.4  333.33
  5367.4  333.75  5368.4  333.71
#Mann= 3 , 1 , 0
 4669.80    0.13       0  4981.6   0.042       0  5018.5    0.13       0
Bank Sta=4981.60,5018.50
Exp/Cntr=0.3,0.1

Type RM Length L Ch R = 1 ,211837.7,727.6,727.6,727.6
BEGIN DESCRIPTION:
Sandy Creek 212.0
END DESCRIPTION:
#Sta/Elev= 20
  4428.4  328.35  4588.4  317.07  4678.4  311.55  4708.4  311.45  4758.4  308.59
  4788.4  307.85  4808.4  305.88  4898.4  300.56  4908.4  300.76  4928.4  299.18
  4976.9  298.88  4979.9  292.88  5020.1  292.88  5023.1  298.88  5060.5  298.92
  5100.5  306.61  5120.5  311.04  5190.5   320.7  5260.5  327.49  5287.7  328.66
#Mann= 3 , 1 , 0
 4428.40    0.13       0  4976.9   0.042       0  5023.1    0.13       0
Bank Sta=4976.90,5023.10
Exp/Cntr=0.3,0.1

Type RM Length L Ch R = 1 ,211110.1,1176.9,1176.9,1176.9
BEGIN DESCRIPTION:
Sandy Creek 211.0
END DESCRIPTION:
#Sta/Elev= 23
  4401.9  329.99  4461.9   327.1  4561.9  319.22  4571.9  317.93  4681.9  310.76
  4711.9  309.79  4731.9  308.43  4861.9  305.89  4921.9  302.47  4931.9  303.86
  4941.9  298.84  4976.9  298.78  4979.9  292.78  5020.1  292.78  5023.1  298.78
  5046.6  298.89  5066.6  302.62  5086.6  308.36  5116.6  315.81  5136.6  319.22
  5166.6  325.69  5176.6  327.47  5189.7  328.23
#Mann= 3 , 1 , 0
 4401.90    0.13       0  4976.9   0.042       0  5023.1    0.13       0
Bank Sta=4976.90,5023.10
Exp/Cntr=0.3,0.1

Type RM Length L Ch R = 1 ,209933.2,23,23,23
BEGIN DESCRIPTION:
Upstream Section of Bridge/Culvert/Weir
END DESCRIPTION:
#Sta/Elev= 25
    4683  311.42  4684.1  311.41    4703  311.27    4723  310.03  4724.1  309.88
    4733  308.64    4743   306.7  4744.1  306.55    4753   305.3  4764.1  305.11
    4783  304.78  4794.1  303.28    4803  302.08    4823     302    4853  296.29
    4904  293.13  4999.9  289.13  5000.1  289.13    5089  293.13    5100  295.25
    5110  301.07  5116.8  302.12    5120  302.61    5160  305.81    5180  306.61
#Mann= 3 , 1 , 0
 4683.00    0.13       0    4904   0.045       0    5089    0.13       0
#XS Ineff= 2 , 0
       0    4893     297    5100       0     297
Bank Sta=4904.00,5089.00
Exp/Cntr=0.5,0.3

Type RM Length L Ch R = 5 ,209921.7,,,
BEGIN DESCRIPTION:
Dam_Southerland Mill Rd_2
Structure ID: Dam_Southerland Mill Rd
Approximate Survey Structure
END DESCRIPTION:
#Inline Weir SE= 25
    4683  311.37  4684.1  311.95    4703  311.23    4723  309.99  4724.1  309.84
    4733  308.77    4743  307.71  4744.1  307.59    4753  305.73  4764.1  305.07
    4783  304.74  4794.1  303.24    4803  302.04    4823  301.96    4853   301.1
    4904  301.49  4999.9  302.23  5000.1  302.24    5089  302.92    5100  303.01
    5110  303.09  5116.8  303.14    5120  302.56    5160  305.76    5180  306.56
IW Dist,WD,Coef,Skew,MaxSub,Min_El,Is_Ogee,SpillHt,DesHd
10.0,3.0,3.0,,0.95,, 0 ,,,2.0,2.0,

Type RM Length L Ch R = 1 ,209910.2,299,299,299
BEGIN DESCRIPTION:
Downstream Section of Bridge/Culvert/Weir
END DESCRIPTION:
#Sta/Elev= 25
    4683  311.31  4684.1   311.3    4703  311.16    4723  309.92  4724.1  309.77
    4733  308.53    4743  306.59  4744.1  306.44    4753  305.19  4764.1     305
    4783  304.67  4794.1  303.17    4803  301.97    4823  301.89    4853  296.18
    4904  293.02  4999.9  289.02  5000.1  289.02    5089  293.02    5100  295.14
    5110  300.96  5116.8  302.01    5120   302.5    5160   305.7    5180   306.5
#Mann= 3 , 1 , 0
 4683.00    0.13       0    4904   0.045       0    5089    0.13       0
#XS Ineff= 2 , 0
       0    4893     297    5100       0     297
Bank Sta=4904.00,5089.00
Exp/Cntr=0.5,0.3

Type RM Length L Ch R = 1 ,209611.2,40,40,40
BEGIN DESCRIPTION:
Upstream Section of Bridge/Culvert/Weir
END DESCRIPTION:
#Sta/Elev= 30
  4644.6  311.79    4661  309.65    4691  307.46    4821  299.37    4861  300.86
    4871  296.86    4941  294.87    4951  293.43    4961   289.5  4977.5  284.62
  4988.5  278.62  5011.5  278.62  5022.5  284.62  5024.1  290.82  5034.1  291.31
  5074.1   300.6  5094.1  302.44  5114.1   301.6  5134.1  302.91  5174.1  303.19
  5204.1  302.34  5234.1  303.52    5296  304.39  5348.6  304.64  5368.6  303.78
  5398.6  304.58  5418.6   306.7  5428.6  305.84  5488.6  308.06  5533.7  311.62
#Mann= 3 , 1 , 0
 4644.60    0.13       0  4977.5   0.045       0  5022.5    0.13       0
#XS Ineff= 2 , 0
       0    4938  301.99    5056       0   302.4
Bank Sta=4977.50,5022.50
Exp/Cntr=0.5,0.3

Type RM Length L Ch R = 3 ,209591.2,,,
BEGIN DESCRIPTION:
Southerland Mill Rd-TOR
Structure ID: Southerland Mill Rd
Approximate Survey Structure
END DESCRIPTION:
Bridge Culvert--1,0,-1,-1, 0
Deck Dist Width WeirC Skew NumUp NumDn MinLoCord MaxHiCord MaxSubmerge Is_Ogee
10,20,2.6,,60,60,,,0.95,0,1,1,,
  4644.6    4661  4664.6  4674.6  4684.6    4691  4704.6  4724.6  4744.6  4814.6
    4821    4831    4861  4864.6    4871    4941 4949.41  4949.5    4951  4957.5
    4961    4971  4977.5  4988.5  5011.5  5022.5  5024.1  5034.1  5039.5  5044.1
 5045.39  5045.5  5054.1  5064.1  5074.1  5094.1  5114.1  5124.1  5134.1  5174.1
  5184.1  5194.1  5204.1  5214.1  5234.1  5244.1  5254.1  5278.6  5288.6    5296
    5326    5336  5348.6    5356  5368.6  5398.6  5418.6  5428.6  5488.6  5533.7
  311.79  309.66   309.4  308.94  309.49  308.78  307.26   306.2  306.26  302.07
  302.06  302.05  302.01     302  302.01  302.16  302.18  302.18  302.18   302.2
  302.21  302.23  302.24  302.26  302.31  302.34  302.34  302.36  302.37  302.38
  302.39  302.39   302.4  302.43  302.45  302.49  302.53  302.55  302.92   303.2
  302.85  303.08  302.72  302.75  303.53  303.65  303.08  303.81  304.36   304.4
  305.34  305.67   305.6  305.56  303.78  304.58   306.7  305.84  308.06  311.62
  311.79  309.65  309.39  308.66  307.93  307.46  306.61  305.37  304.12  299.77
  299.37  299.48  300.86  299.42  296.86  294.87  293.66  299.38  299.38   299.4
  299.41  299.43  299.44  299.46  299.51  299.54  299.54  299.56  299.57  299.58
  299.59  293.72  296.02  297.95   300.6  302.44   301.6  301.88  302.91  303.19
  302.84  303.07  302.34  302.47  303.52  303.64  303.07   303.8  304.35  304.39
  304.53  304.58  304.64  304.32  303.78  304.58   306.7  305.84  308.06  311.62
  4644.6    4661  4664.6  4674.6  4684.6    4691  4704.6  4724.6  4744.6  4814.6
    4821    4831    4861  4864.6    4871    4941 4949.41  4949.5    4951  4957.5
    4961    4971  4977.5  4988.5  5011.5  5022.5  5024.1  5034.1  5039.5  5044.1
 5045.39  5045.5  5054.1  5064.1  5074.1  5094.1  5114.1  5124.1  5134.1  5174.1
  5184.1  5194.1  5204.1  5214.1  5234.1  5244.1  5254.1  5278.6  5288.6    5296
    5326    5336  5348.6    5356  5368.6  5398.6  5418.6  5428.6  5488.6  5533.7
  311.79  309.66   309.4  308.94  309.49  308.78  307.26   306.2  306.26  302.07
  302.06  302.05  302.01     302  302.01  302.16  302.18  302.18  302.18   302.2
  302.21  302.23  302.24  302.26  302.31  302.34  302.34  302.36  302.37  302.38
  302.39  302.39   302.4  302.43  302.45  302.49  302.53  302.55  302.92   303.2
  302.85  303.08  302.72  302.75  303.53  303.65  303.08  303.81  304.36   304.4
  305.34  305.67   305.6  305.56  303.78  304.58   306.7  305.84  308.06  311.62
  311.79  309.65  309.39  308.66  307.93  307.46  306.61  305.37  304.12  299.77
  299.37  299.48  300.86  299.42  296.86  294.87  293.66  299.38  299.38   299.4
  299.41  299.43  299.44  299.46  299.51  299.54  299.54  299.56  299.57  299.58
  299.59  293.72  296.02  297.95   300.6  302.44   301.6  301.88  302.91  303.19
  302.84  303.07  302.34  302.47  303.52  303.64  303.07   303.8  304.35  304.39
  304.53  304.58  304.64  304.32  303.78  304.58   306.7  305.84  308.06  311.62
Pier Skew, UpSta & Num, DnSta & Num=,4966.0, 2 ,4966.0, 2 , 0 , 0 , 0 ,,
     1.5     1.5
  286.95  300.42
     1.5     1.5
  286.95  300.42
Pier Skew, UpSta & Num, DnSta & Num=,4983.0, 2 ,4983.0, 2 , 0 , 0 , 0 ,,
     1.5     1.5
  280.21  300.45
     1.5     1.5
  280.21  300.45
Pier Skew, UpSta & Num, DnSta & Num=,5000.0, 2 ,5000.0, 2 , 0 , 0 , 0 ,,
     1.5     1.5
  277.62  300.49
     1.5     1.5
  277.62  300.49
Pier Skew, UpSta & Num, DnSta & Num=,5017.0, 2 ,5017.0, 2 , 0 , 0 , 0 ,,
     1.5     1.5
  280.21  300.53
     1.5     1.5
  280.21  300.53
Pier Skew, UpSta & Num, DnSta & Num=,5034.0, 2 ,5034.0, 2 , 0 , 0 , 0 ,,
     1.5     1.5
  290.27  300.56
     1.5     1.5
  290.27  300.56
Abutment Skew #Up #Dn=, 2 , 2
 4949.30 4957.50
  299.38  290.88
 4949.30 4957.50
  299.38  290.88
Abutment Skew #Up #Dn=, 2 , 2
 5039.50 5045.59
  292.41  299.59
 5039.50 5045.59
  292.41  299.59
BR Coef= 1 , 1 , 0 ,1.25, 0 ,,,0.8,0,2,0,
Wspro=,,,, 1 ,,,, 0 ,,,, 0 ,,,,-1 ,-1 ,-1 , 0 , 0 , 0 , 0 , 0
BC Design=,, 0 ,, 0 ,,,,,,
BR U #Sta/Elev= 60
  4644.6  311.79    4661  309.65  4664.6  309.39  4674.6  308.66  4684.6  307.93
    4691  307.46  4704.6  306.61  4724.6  305.37  4744.6  304.12  4814.6  299.77
    4821  299.37    4831  299.48    4861  300.86  4864.6  299.42    4871  296.86
    4941  294.87 4949.41  293.66  4949.5  293.65    4951  293.43  4957.5  290.88
    4961   289.5    4971   286.8  4977.5  284.62  4988.5  278.62  5011.5  278.62
  5022.5  284.62  5024.1  290.82  5034.1  291.31  5039.5  292.41  5044.1  293.35
 5045.39  293.69  5045.5  293.72  5054.1  296.02  5064.1  297.95  5074.1   300.6
  5094.1  302.44  5114.1   301.6  5124.1  301.88  5134.1  302.91  5174.1  303.19
  5184.1  302.84  5194.1  303.07  5204.1  302.34  5214.1  302.47  5234.1  303.52
  5244.1  303.64  5254.1  303.07  5278.6   303.8  5288.6  304.35    5296  304.39
    5326  304.53    5336  304.58  5348.6  304.64    5356  304.32  5368.6  303.78
  5398.6  304.58  5418.6   306.7  5428.6  305.84  5488.6  308.06  5533.7  311.62
BR U #Mann= 3
 4644.60    0.13  4977.5   0.045  5022.5    0.13
BR U Banks=4977.50,5022.50
BR D #Sta/Elev= 60
  4644.6  311.79    4661  309.65  4664.6  309.39  4674.6  308.66  4684.6  307.93
    4691  307.46  4704.6  306.61  4724.6  305.37  4744.6  304.12  4814.6  299.77
    4821  299.37    4831  299.48    4861  300.86  4864.6  299.42    4871  296.86
    4941  294.87 4949.41  293.66  4949.5  293.65    4951  293.43  4957.5  290.88
    4961   289.5    4971   286.8  4977.5  284.62  4988.5  278.62  5011.5  278.62
  5022.5  284.62  5024.1  290.82  5034.1  291.31  5039.5  292.41  5044.1  293.35
 5045.39  293.69  5045.5  293.72  5054.1  296.02  5064.1  297.95  5074.1   300.6
  5094.1  302.44  5114.1   301.6  5124.1  301.88  5134.1  302.91  5174.1  303.19
  5184.1  302.84  5194.1  303.07  5204.1  302.34  5214.1  302.47  5234.1  303.52
  5244.1  303.64  5254.1  303.07  5278.6   303.8  5288.6  304.35    5296  304.39
    5326  304.53    5336  304.58  5348.6  304.64    5356  304.32  5368.6  303.78
  5398.6  304.58  5418.6   306.7  5428.6  305.84  5488.6  308.06  5533.7  311.62
BR D #Mann= 3
 4644.60    0.13  4977.5   0.045  5022.5    0.13
BR D Banks=4977.50,5022.50

Type RM Length L Ch R = 1 ,209571.2,384.1,384.1,384.1
BEGIN DESCRIPTION:
Downstream Section of Bridge/Culvert/Weir
END DESCRIPTION:
#Sta/Elev= 30
  4644.6  311.79    4661  309.65    4691  307.46    4821  299.37    4861  300.86
    4871  296.86    4941  294.87    4951  293.43    4961   289.5  4977.5  284.62
  4988.5  278.62  5011.5  278.62  5022.5  284.62  5024.1  290.82  5034.1  291.31
  5074.1   300.6  5094.1  302.44  5114.1   301.6  5134.1  302.91  5174.1  303.19
  5204.1  302.34  5234.1  303.52    5296  304.39  5348.6  304.64  5368.6  303.78
  5398.6  304.58  5418.6   306.7  5428.6  305.84  5488.6  308.06  5533.7  311.62
#Mann= 3 , 1 , 0
 4644.60    0.13       0  4977.5   0.045       0  5022.5    0.13       0
#XS Ineff= 2 , 0
       0    4938  301.99    5056       0   302.4
Bank Sta=4977.50,5022.50
Exp/Cntr=0.5,0.3

Type RM Length L Ch R = 1 ,209187.1,936.2,936.2,936.2
BEGIN DESCRIPTION:
Sandy Creek 209.0
END DESCRIPTION:
#Sta/Elev= 23
  4712.9  321.92  4762.9  314.05  4782.9   312.3  4822.9  307.21  4832.9  306.46
  4852.9  303.66  4902.9  294.21  4922.9  292.46  4942.9  292.26  4952.9  291.44
  4972.9  287.54  4976.9  284.58  4979.9  278.58  5020.1  278.58  5023.1  284.58
  5050.9  291.47  5080.9  292.25  5150.9  298.56  5180.9  299.88  5210.9  302.86
  5260.9  308.81  5390.9  315.38  5458.6  317.72
#Mann= 3 , 1 , 0
 4712.90    0.13       0  4976.9   0.042       0  5023.1    0.13       0
Bank Sta=4976.90,5023.10
Exp/Cntr=0.3,0.1

Type RM Length L Ch R = 1 ,208250.9,1113.5,1113.5,1113.5
BEGIN DESCRIPTION:
Sandy Creek 208.0
END DESCRIPTION:
#Sta/Elev= 26
  4505.3  321.43  4575.3  315.88  4615.3  313.07  4685.3  305.88  4705.3  304.89
  4775.3  297.25  4805.3  296.45  4835.3  291.52  4845.3  290.89  4865.3  287.69
  4875.3  289.18  4885.3  291.47  4895.3  291.59  4905.3  293.57  4915.3  293.51
  4925.3   292.2  4965.3  291.23  4975.3   291.3  4976.9  284.49  4979.9  278.49
  5020.1  278.49  5023.1  284.49  5032.6  288.78  5042.6  295.38  5072.6  309.08
  5119.5  317.65
#Mann= 3 , 1 , 0
 4505.30    0.13       0  4976.9   0.042       0  5023.1    0.13       0
Bank Sta=4976.90,5023.10
Exp/Cntr=0.3,0.1

Type RM Length L Ch R = 1 ,207137.4,1016.7,1016.7,1016.7
BEGIN DESCRIPTION:
Sandy Creek 207.0
END DESCRIPTION:
#Sta/Elev= 30
  4554.9  334.09  4594.9  331.14  4654.9  328.29  4684.9  325.19  4764.9  315.27
  4854.9  297.21  4874.9  292.27  4924.9  289.39  4934.9  289.56  4954.9  291.39
  4964.9  290.63  4974.9  288.67  4975.2  284.38  4978.2  278.38  5021.9  278.38
  5024.9  284.38  5033.9  290.93  5043.9  291.56  5063.9  295.94  5083.9  298.99
  5103.9  299.92  5133.9  298.77  5153.9  300.27  5173.9  305.04  5183.9  306.26
  5203.9  306.26  5243.9  308.08  5283.9  312.15  5293.9  312.38  5338.6  317.85
#Mann= 3 , 1 , 0
 4554.90    0.13       0  4975.2   0.042       0  5024.9    0.13       0
Bank Sta=4975.20,5024.90
Exp/Cntr=0.3,0.1

Type RM Length L Ch R = 1 ,206120.7,1371.6,1371.6,1371.6
BEGIN DESCRIPTION:
Sandy Creek 206.0
END DESCRIPTION:
#Sta/Elev= 30
  4520.3  317.24  4590.3  311.42  4650.3  304.66  4680.3     300  4740.3  294.56
  4840.3  289.36  4900.3  288.42  4920.3  289.36  4960.3  289.57  4970.3  288.07
  4975.1  282.57  4978.1  276.57  5021.8  276.57  5024.8  282.57  5030.3  289.64
  5050.3  290.67  5070.3  288.39  5080.3  288.73  5090.3  290.16  5200.3  293.51
  5220.3  296.93  5240.3  302.76  5250.3  303.76  5270.3  303.27  5290.3  305.17
  5370.3  304.48  5390.3  306.31  5410.3  304.78  5470.3  309.85    5510  311.86
#Mann= 3 , 1 , 0
 4520.30    0.13       0  4975.1   0.042       0  5024.8    0.13       0
Bank Sta=4975.10,5024.80
Exp/Cntr=0.3,0.1

Type RM Length L Ch R = 1 ,204749.1,1089.4,1089.4,1089.4
BEGIN DESCRIPTION:
Sandy Creek 205.0
END DESCRIPTION:
#Sta/Elev= 30
  4263.8  331.31  4283.8  328.36  4393.8  318.25  4513.8  303.85  4593.8  300.89
  4743.8  299.08  4793.8   297.9  4833.8  295.61  4893.8  294.63  4923.8  292.56
  4973.8  281.89  4975.2  281.04  4978.2  275.04  5021.9  275.04  5024.9  281.04
  5043.7  288.47  5053.7  287.64  5133.7  287.68  5213.7  285.82  5233.7   287.4
  5343.7  287.66  5373.7  285.91  5413.7  288.23  5463.7  289.74  5503.7  289.89
  5513.7  290.87  5533.7  295.53  5553.7  301.82  5583.7  313.03  5604.2  319.74
#Mann= 3 , 1 , 0
 4263.80    0.13       0  4975.2   0.042       0  5024.9    0.13       0
Bank Sta=4975.20,5024.90
Exp/Cntr=0.3,0.1

Type RM Length L Ch R = 1 ,203659.7,1847,1847,1847
BEGIN DESCRIPTION:
Sandy Creek 203.0
END DESCRIPTION:
#Sta/Elev= 30
  4280.7  310.79  4320.7  310.16  4490.7  302.73  4620.7  299.63  4890.7  296.93
  4910.7  295.65  4970.7  287.81  4975.1  280.44  4978.1  274.44  5021.9  274.44
  5024.9  280.44  5026.3   287.2  5126.3   284.6  5226.3  285.38  5246.3  283.65
  5266.3  284.84  5366.3  284.18  5396.3   285.4  5416.3  284.48  5499.9  284.37
  5566.3  284.95  5586.3  283.56  5606.3  284.77  5666.3  284.63  5716.3     286
  5806.3  284.31  5826.3  289.87  5856.3  302.52  5886.3  310.25  5932.8  317.47
#Mann= 4 , 1 , 0
 4280.70    0.13       0  4975.1   0.042       0  5024.9    0.13       0
  5499.9       1       0
Bank Sta=4975.10,5024.90
Exp/Cntr=0.3,0.1

Type RM Length L Ch R = 1 ,201812.7,972.2,972.2,972.2
BEGIN DESCRIPTION:
Sandy Creek 202.0
END DESCRIPTION:
#Sta/Elev= 30
  4462.4  311.08  4852.4  288.59  4952.4  286.62  4972.4  285.29  4975.2  277.94
  4978.2  271.94  5021.9  271.94  5024.9  277.94  5028.7  283.95  5108.7  282.25
  5128.7  283.21  5218.7   281.2  5238.7  282.32  5278.7  281.08  5308.7   283.6
  5398.7  280.29  5428.7  281.92  5499.9  281.78  5518.7  283.03  5538.7  281.41
  5668.7  282.27  5738.7  280.75  5948.7  281.83  6028.7  281.15  6058.7  282.43
  6128.7  283.04  6178.7  285.48  6188.7   287.1  6268.7  307.72  6344.2  319.72
#Mann= 4 , 1 , 0
 4462.40    0.13       0  4975.2   0.042       0  5024.9    0.13       0
  5499.9       1       0
Bank Sta=4975.20,5024.90
Exp/Cntr=0.3,0.1

Type RM Length L Ch R = 1 ,200840.5,1430.1,1430.1,1430.1
BEGIN DESCRIPTION:
Sandy Creek 201.0
END DESCRIPTION:
#Sta/Elev= 30
  4409.4  311.51  4439.4  309.86  4469.4  309.11  4479.4  308.31  4489.4   306.9
  4569.4  301.46  4599.4  296.79  4679.4  288.03  4719.4   281.3  4729.4  280.37
  4879.4  280.63  4909.4  283.02  4959.4  284.12  4969.4  283.15    4974  276.51
    4977  270.51    5023  270.51    5026  276.51  5050.5  282.84  5060.5  283.13
  5080.5  282.36  5100.5  282.62  5160.5  281.26  5220.5  282.16  5280.5   285.6
  5320.5  290.13  5350.5  295.18  5400.5  300.78  5450.5  304.92  5494.3   306.5
#Mann= 3 , 1 , 0
 4409.40    0.13       0    4974   0.042       0    5026    0.13       0
Bank Sta=4974.00,5026.00
Exp/Cntr=0.3,0.1

Type RM Length L Ch R = 1 ,199410.4,1204.8,1204.8,1204.8
BEGIN DESCRIPTION:
Sandy Creek 199.0
END DESCRIPTION:
#Sta/Elev= 30
  3862.2  313.03  3942.2  301.92  3982.2  298.75  4042.2  296.64  4192.2  295.39
  4332.2  291.59  4362.2   289.2  4392.2  288.57  4462.2  290.11  4552.2  289.61
  4642.2  286.41  4702.2  281.99  4712.2  279.85  4732.2  282.41  4762.2  283.62
  4792.2  281.31  4902.2  281.05  4972.2  282.14    4974  274.22    4977  268.22
    5023  268.22    5026  274.22  5037.1  279.18  5047.1  279.78  5147.1  278.02
  5157.1  279.11  5247.1  280.86  5267.1  283.04  5287.1  291.15  5388.4  313.27
#Mann= 3 , 1 , 0
 3862.20    0.13       0    4974   0.042       0    5026    0.13       0
Bank Sta=4974.00,5026.00
Exp/Cntr=0.3,0.1

Type RM Length L Ch R = 1 ,198205.6,1216,1216,1216
BEGIN DESCRIPTION:
Sandy Creek 198.0
END DESCRIPTION:
#Sta/Elev= 28
  4114.4  310.29  4214.4  306.68  4554.4  292.68  4664.4  291.27  4724.4  286.93
  4764.4  280.96  4794.4   279.1  4824.4  276.23  4894.4  278.13  4904.4  278.96
  4954.4  280.24    4974  273.45    4977  267.45    5023  267.45    5026  273.45
  5035.7  279.26  5055.7  280.08  5085.7  278.55  5095.7  277.69  5115.7  277.68
  5125.7  277.06  5135.7  277.44  5155.7  276.77  5165.7  276.84  5185.7  277.68
  5225.7  294.19  5265.7  308.32  5310.7  319.59
#Mann= 3 , 1 , 0
 4114.40    0.13       0    4974   0.042       0    5026    0.13       0
Bank Sta=4974.00,5026.00
Exp/Cntr=0.3,0.1

Type RM Length L Ch R = 1 ,196989.6,1507.4,1507.4,1507.4
BEGIN DESCRIPTION:
Sandy Creek 197.0
END DESCRIPTION:
#Sta/Elev= 30
  3621.7   315.7  3761.7  310.45  3841.7  301.77  3911.7  298.42  3941.7  293.08
  4041.7  281.98  4261.7  280.94  4311.7   282.1  4331.7  280.69  4521.7  277.93
  4811.7  276.25  4971.7  276.71    4974  272.67    4977  266.67    5023  266.67
    5026  272.67    5030  276.02    5050  277.12    5140  278.54    5180  277.08
    5210  278.25  5499.9  276.07    5640  276.89    5930  283.06    5940  285.51
    6010  294.69    6040   300.3    6060  302.75    6130  307.98  6194.2  314.71
#Mann= 4 , 1 , 0
 3621.70    0.13       0    4974   0.042       0    5026    0.13       0
  5499.9       1       0
Bank Sta=4974.00,5026.00
Exp/Cntr=0.3,0.1

Type RM Length L Ch R = 1 ,195482.2,1139,1139,1139
BEGIN DESCRIPTION:
Sandy Creek 195.0
END DESCRIPTION:
#Sta/Elev= 30
  4058.9  302.56  4088.9  298.21  4108.9  296.85  4128.9  292.97  4198.9   287.9
  4258.9  281.94  4388.9  275.85  4448.9  274.47  4518.9  275.36  4888.9  274.78
    4974  271.71    4977  265.71    5023  265.71    5026  271.71  5032.9  275.12
  5112.9  276.85  5132.9  278.58  5162.9  278.65  5212.9  275.72  5302.9  284.02
  5342.9  285.24  5392.9  284.09  5692.9  284.94  5792.9  283.15  5852.9  284.02
  5922.9  287.67  6012.9  295.16  6052.9  295.95  6112.9  302.74  6224.8  309.02
#Mann= 3 , 1 , 0
 4058.90    0.13       0    4974   0.042       0    5026    0.13       0
Bank Sta=4974.00,5026.00
Exp/Cntr=0.3,0.1

Type RM Length L Ch R = 1 ,194343.2,1220.9,1220.9,1220.9
BEGIN DESCRIPTION:
Sandy Creek 194.0
END DESCRIPTION:
#Sta/Elev= 30
  3947.2  298.71  4257.2  289.42  4367.2  287.93  4507.2  284.47  4547.2  284.59
  4557.2   283.5  4677.2  279.35  4767.2  278.25  4827.2  278.89  4907.2  275.01
  4937.2  272.53  4967.2  273.64  4972.9  270.98  4975.9  264.98  5024.2  264.98
  5027.2  270.98  5037.7  275.31  5057.7  275.82  5227.7  272.18  5247.7  273.42
  5307.7  272.25  5347.7  273.06  5367.7  271.87  5447.7  273.41  5627.7  279.91
  5657.7  281.96  5727.7  289.07  5867.7  306.39  5927.7  310.71    5974  312.86
#Mann= 3 , 1 , 0
 3947.20    0.13       0  4972.9   0.042       0  5027.2    0.13       0
Bank Sta=4972.90,5027.20
Exp/Cntr=0.3,0.1

Type RM Length L Ch R = 1 ,193122.3,1133,1133,1133
BEGIN DESCRIPTION:
Sandy Creek 193.0
END DESCRIPTION:
#Sta/Elev= 30
  4352.3  295.41  4532.3  285.04  4572.3  280.59  4592.3  277.51  4632.3  273.81
  4672.3  272.13  4692.3  273.03  4712.3     272  4802.3  273.19  4902.3   272.3
  4942.3  273.47  4972.8   270.2  4975.8   264.2  5024.1   264.2  5027.1   270.2
  5029.7  273.73  5099.7  273.46  5159.7  274.27  5199.7  273.08  5229.7   274.8
  5289.7  273.67  5359.7  275.29  5429.7  281.52  5469.7  288.87  5489.7  289.42
  5519.7   293.9  5539.7  293.74  5579.7  299.55  5669.7   308.5  5724.6  310.56
#Mann= 3 , 1 , 0
 4352.30    0.13       0  4972.8   0.042       0  5027.1    0.13       0
Bank Sta=4972.80,5027.10
Exp/Cntr=0.3,0.1

Type RM Length L Ch R = 1 ,191989.3,870.7,870.7,870.7
BEGIN DESCRIPTION:
Sandy Creek 192.0
END DESCRIPTION:
#Sta/Elev= 30
  4075.6  295.55  4095.6  294.17  4145.6  286.73  4195.6  281.07  4255.6  276.71
  4305.6  275.61  4345.6  272.52  4375.6   271.8  4435.6  272.94  4499.9  272.27
  4655.6  273.66  4705.6   272.1  4935.6  272.66  4955.6  272.15  4972.9  269.47
  4975.9  263.47  5024.1  263.47  5027.1  269.47    5070  271.93    5150  273.08
    5230  271.12    5330  272.72    5410  271.23  5499.9  272.53    5640  274.86
    5660  280.08    5670  284.08    5690  297.16    5700  302.04  5759.3  319.69
#Mann= 5 , 1 , 0
 4075.60       1       0  4499.9    0.13       0  4972.9   0.042       0
  5027.1    0.13       0  5499.9       1       0
Bank Sta=4972.90,5027.10
Exp/Cntr=0.3,0.1

Type RM Length L Ch R = 1 ,191118.6,971.8,971.8,971.8
BEGIN DESCRIPTION:
Sandy Creek 191.0
END DESCRIPTION:
#Sta/Elev= 30
  4306.8  296.77  4366.8  295.65  4406.8  293.44  4416.8  292.14  4466.8  289.31
  4546.8   281.2  4596.8  279.29  4616.8   280.2  4696.8  272.14  4736.8  270.33
  4816.8  271.66  4846.8  270.48  4972.9  268.92  4975.9  262.92  5024.2  262.92
  5027.2  268.92    5139  270.78    5179  269.34    5249  270.35    5279  269.91
    5349  270.34    5369  269.63    5419  269.95    5429  270.39    5449  272.72
    5459   275.9    5489  286.75    5499  289.73    5549  297.52  5563.1  298.92
#Mann= 3 , 1 , 0
 4306.80    0.13       0  4972.9   0.042       0  5027.2    0.13       0
Bank Sta=4972.90,5027.20
Exp/Cntr=0.3,0.1

Type RM Length L Ch R = 1 ,190146.8,38,38,38
BEGIN DESCRIPTION:
Upstream Section of Bridge/Culvert/Weir
END DESCRIPTION:
#Sta/Elev= 30
    3861  306.46  4097.7  285.68  4157.7  281.41  4227.7  282.01  4257.7  280.03
  4287.7  276.85  4357.7  274.05  4367.7  274.52  4417.7  270.52  4437.7  271.12
  4467.7  270.44  4499.9  270.63  4617.7  271.33  4637.7  269.63  4717.7  273.22
  4727.7  272.79  4817.7  274.26  4907.7  271.21  4927.7  274.04  4982.5  268.29
  4984.5  262.29  5015.5  262.29  5017.5  268.29  5026.7  272.44  5156.7  274.25
  5276.7  280.18  5306.7  280.73  5356.7  283.75  5376.7  284.26  5587.8  302.86
#Mann= 4 , 1 , 0
 3861.00       1       0  4499.9    0.13       0  4982.5   0.042       0
  5017.5    0.13       0
#XS Ineff= 2 , 0
       0    4974  271.86    5026       0  273.84
Bank Sta=4982.50,5017.50
Exp/Cntr=0.5,0.3
